--- SFTOMLINRN.prj (project) ---

Proj Title=SFTOMLINRN
Current Plan=p01
Default Exp/Contr=0,0
English Units
Geom File=g01
Flow File=f01
Plan File=p01
BEGIN DESCRIPTION:
END DESCRIPTION:
DSS Export Rating Curves= 0
DSS Export Rating Curve Sorted= 0
DSS Export Volume Flow Curves= 0
DXF Filename=..\..\..\..\..\Engineering\Hydraulics\SFTOMLINRN\SFTOMLINRN.
DXF OffsetX= 0
DXF OffsetY= 0
DXF ScaleX= 0
DXF ScaleY= 0

--- SFTOMLINRN.p01 (plan) ---

Plan Title=Floodplain
Program Version=4.00
Geom File=g01
Flow File=f01
K Sum by GR=0
Std Step Tol=0.01
Critical Tol=0.01
Num of Std Step Trials=20
Max Error Tol=0.3
Flow Tol Ratio=0.001
Split Flow NTrial=30
Split Flow Tol=0.02
Split Flow Ratio=0.02
Log Output Level=0
Friction Slope Method=1
Unsteady Friction Slope Method=2
Unsteady Bridges Friction Slope Method=1
Global Log Level=0
CheckData=False
Run HTab=0
Run UNet=0
Run PostProcess=0
UNET Theta=0
UNET Theta Warmup=0
UNET ZTol=0
UNET ZSATol=0
UNET MxIter=0
UNET MaxInSteps=0
UNET DtIC=0
UNET DtMin=0
UNET MaxCRTS=0
UNET WFStab=0
UNET SFStab=0
UNET WFX=0
UNET SFX=0
UNET DSS MLevel=0
UNET DZMax Abort=0
UNET Convert EG Bridges=0
UNET Use Existing IB Tables=0
UNET Froude Limit=0
UNET Froude Power=0
Write IC File=0
Echo Input=False
Echo Output=False
Write Detailed=0

--- SFTOMLINRN.f01 (steady flow) ---

Flow Title=NFF Regression Equation
Program Version=4.10
Number of Profiles= 1
Profile Names=P100yr
River Rch & RM=SFTOMLINRN,Main            ,32281.2
  1170.6
River Rch & RM=SFTOMLINRN,Main            ,30984.6
    1256
River Rch & RM=SFTOMLINRN,Main            ,29148.6
    1320
River Rch & RM=SFTOMLINRN,Main            ,26822.4
1577.587
River Rch & RM=SFTOMLINRN,Main            ,23662.1
1668.347
River Rch & RM=SFTOMLINRN,Main            ,23180
1850.413
River Rch & RM=SFTOMLINRN,Main            ,20797.7
1871.885
River Rch & RM=SFTOMLINRN,Main            ,20500.7
2141.984
River Rch & RM=SFTOMLINRN,Main            ,15422
 2350.09
River Rch & RM=SFTOMLINRN,Main            ,8933.4
2580.791
River Rch & RM=SFTOMLINRN,Main            ,283.7
2848.541
Boundary for River Rch & Prof#=SFTOMLINRN,Main            , 1
Up Type= 0
Dn Type= 1
Dn Known WS=918.81
DSS Import GetInterval= 0
DSS Import GetPeak= 0
DSS Import FillOption= 0

--- SFTOMLINRN.g01 (geometry) ---

Geom Title=2003 WVU SAMB 3 Meter DEM
Program Version=4.10

River Reach=SFTOMLINRN      ,Main
Reach XY= 30
     1685326.056      749277.136     1684749.233      748853.959
     1684363.816      747546.667     1684193.243       744866.98
     1683478.846      743806.845     1682551.135      743598.672
     1681832.207      743540.561      1681215.35      744003.136
     1680607.883       743791.92     1679672.121      744207.123
     1679008.926      743898.095     1678947.294      744090.803
     1678224.204      744085.595     1677942.954      743844.276
     1676075.859      744843.253     1675541.058      744840.923
     1675178.698      745315.136     1674582.144      745322.127
     1673896.079      744731.428     1673756.056      744907.336
     1674020.544       745019.19     1673204.181      745536.425
     1672063.941      745113.468     1671186.444      744218.408
     1670909.164      744517.112     1670347.902      744292.626
     1668500.246      745356.428       1667034.1       744782.21
     1666143.909       746171.75     1665551.799      746110.023

Type RM Length L Ch R = 1 ,32281.2 ,518.2,616.9,621.2
XS GIS Cut Line= 2
     1685260.789      748742.016     1685288.567      749804.516
#Sta/Elev= 30
       0 1125.55    39.4 1118.89      59  1116.3    88.6 1115.92    98.4 1115.27
   127.9 1111.56   177.1 1106.34   265.7 1099.14   295.2 1096.16   334.6 1089.58
   403.5 1079.83     433  1075.2   472.4 1067.89   492.1 1065.84   521.6 1065.09
   541.3 1064.38   552.41064.638   580.6 1066.22   629.8  1066.8   698.7 1069.85
   708.6  1069.6   718.4 1067.06   728.3  1066.6   747.9 1066.91   767.6 1068.81
   797.2 1070.87   925.1 1089.36     994 1098.09  1013.7 1099.98  1062.9 1103.25
#Mann= 3 , 0 , 0
       0      .1       0   521.6    .045       0   552.4     .06       0
#XS Ineff= 2 , 0
                          700.14         1072.14
Permanent Ineff=
       F       F
Bank Sta=521.6,552.4
XS Rating Curve= 0 ,0
Exp/Cntr=0.3,0.1

Type RM Length L Ch R = 1 ,31664.3 ,476.1,455.5,436.8
XS GIS Cut Line= 4
     1685222.594      748870.488     1685094.122      748971.183
     1684847.594      749151.738     1684729.539      749245.488
#Sta/Elev= 30
       0 1104.83      48 1095.36      96 1085.65     144  1075.6   182.3 1067.09
   191.9 1065.57   201.4 1064.93   220.5 1064.75   268.3 1065.49   277.8 1065.37
   296.9 1064.15     316  1063.9     354  1063.9     3761063.902   382.9 1063.91
   392.4 1064.55   411.5 1067.23   421.1 1067.76   440.2 1068.02   449.7 1068.68
   459.3 1069.94   487.6 1075.27   497.1 1077.18   506.5 1079.37   515.9 1081.77
   534.8 1086.98   581.9 1100.78   591.3  1103.2   600.7 1105.33   619.6 1109.16
#Mann= 3 , 0 , 0
       0     .08       0     354    .045       0     376     .08       0
Bank Sta=354,376
XS Rating Curve= 0 ,0
Exp/Cntr=0.3,0.1

Type RM Length L Ch R = 1 ,31208.8 ,232.5,224.2,216.7
XS GIS Cut Line= 2
     1685135.789       748686.46     1684514.261      749075.349
#Sta/Elev= 30
       0 1103.93    19.6 1100.24    29.3 1098.04    68.4 1087.24      88 1082.01
   117.3 1074.95   127.1 1072.82   146.6 1068.99   156.4 1067.18   166.2 1065.77
     176 1065.03   185.7 1064.84   215.1 1065.54   224.8 1065.58   293.3 1063.99
     303  1063.9   361.7  1063.9     3971063.911   410.6 1064.32   420.4  1065.8
   430.1 1067.65   488.8 1077.23   527.9 1083.04   547.4 1085.44   576.8 1088.44
   615.9 1091.49   645.2 1095.73   684.3 1099.04   713.6 1100.94   733.2 1102.64
#Mann= 3 , 0 , 0
       0     .08       0   361.7    .045       0     397     .07       0
Bank Sta=361.7,397
XS Rating Curve= 0 ,0
Exp/Cntr=0.3,0.1

Type RM Length L Ch R = 1 ,30984.6 ,111.1,111.1,111.1
XS GIS Cut Line= 2
     1685062.872      748519.794     1684361.483      748926.044
#Sta/Elev= 30
       0 1095.51     9.8 1095.21    19.5 1093.77    39.1 1089.19    78.1    1079
    97.7 1074.65   107.4 1072.85     127 1069.92   146.5 1067.79     166 1066.29
   185.6 1065.57   224.6 1065.59   322.3  1063.9     372  1063.9   410.2  1063.9
     459 1064.05   468.8 1064.43   488.3 1066.42     498 1065.84   507.8 1064.77
   517.6 1064.27   527.3  1064.6   546.9 1066.33   556.6 1066.46   576.2 1066.13
   595.7 1066.49   654.3 1069.56   693.4 1070.43   742.2 1072.86   810.6 1075.11
#Mann= 3 , 0 , 0
       0     .07       0     372    .045       0   410.2     .07       0
Bank Sta=372,410.2
XS Rating Curve= 0 ,0
Exp/Cntr=0.3,0.1

Type RM Length L Ch R = 1 ,30873.5 ,297.3,296.3,288.7
XS GIS Cut Line= 2
     1684979.539      748439.933      1684278.15      748846.183
#Sta/Elev= 30
       0 1085.02    29.3 1080.02    58.6 1075.66    97.7 1070.56   107.4 1069.55
   117.2 1068.86   156.2 1066.73   175.8 1065.98   224.6 1065.36   253.9 1065.71
   273.4 1065.21     293 1064.21   312.5  1063.9   333.8  1063.9   361.3 1063.96
   371.1 1064.46   419.9 1069.77   439.4 1071.32     459 1072.12   468.8 1072.23
   527.3  1072.3   546.9 1073.22   595.7 1076.43   605.5 1077.22   634.8 1080.24
   664.1 1082.99   703.1 1085.63   761.7 1091.18   781.2 1092.78   810.6  1094.6
#Mann= 3 , 0 , 0
       0     .08       0   333.8    .045       0   361.3     .07       0
Bank Sta=333.8,361.3
XS Rating Curve= 0 ,0
Exp/Cntr=0.3,0.1

Type RM Length L Ch R = 1 ,30577.2 ,352.7,355.1,355.8
XS GIS Cut Line= 3
     1684944.817      748255.905     1684861.483      748290.627
     1684205.233      748630.905
#Sta/Elev= 30
       0  1093.1    18.1 1087.79    45.1 1079.47    72.2 1071.35    81.2  1068.8
    90.3 1066.46     100  1064.7   109.7    1064   138.9  1063.9   236.2  1063.9
     2701064.139   284.8  1063.9   302.2  1063.9     314    1064   323.7 1064.37
   343.2 1065.65   362.6 1066.63   401.5 1070.14   469.6 1077.26   576.6 1087.35
   596.1 1089.58   615.5 1092.18   664.2 1098.07   703.1 1101.98   722.5 1104.82
     742 1107.94   751.7 1109.69   771.1 1113.88   800.3 1119.36   829.5 1125.56
#Mann= 3 , 0 , 0
       0     .06       0     270    .045       0   302.2     .08       0
Bank Sta=270,302.2
XS Rating Curve= 0 ,0
Exp/Cntr=0.3,0.1

Type RM Length L Ch R = 1 ,30222.1 ,603.2,603.5,603.6
XS GIS Cut Line= 2
     1684851.067      747929.516      1684215.65      748203.821
#Sta/Elev= 30
       0 1091.87     9.8 1091.47    19.5 1090.37    29.2 1088.18   107.2 1065.91
     117 1063.63   126.7 1062.49     156  1062.2   204.7 1062.24   263.2 1063.49
   292.4 1063.56   321.7 1062.57   331.4 1062.51   341.2 1062.77   350.9 1063.68
   360.7 1064.46   380.2 1065.21   399.7 1066.38   428.9 1068.63   497.1 1073.32
   555.6 1077.93   565.4 1078.61   584.9  1079.4   594.6 1080.05   614.1  1081.8
   623.9 1082.18   633.6  1082.2   643.4 1082.54   653.1  1083.2   692.1 1087.42
#Mann= 3 , 0 , 0
       0     .06       0   292.4    .045       0   350.9     .08       0
Bank Sta=292.4,350.9
XS Rating Curve= 0 ,0
Exp/Cntr=0.3,0.1

Type RM Length L Ch R = 1 ,29618.6 ,459.2,470,478.4
XS GIS Cut Line= 2
     1684757.317      747349.655     1684014.261      747676.044
#Sta/Elev= 30
       0 1110.17      88 1089.74    97.8 1087.85   107.6 1086.94   117.3 1086.68
   127.1 1085.68   136.9 1083.56   146.7 1080.98   205.3 1064.74   215.1 1062.84
   224.9 1061.95     264  1059.5   273.8 1059.03   312.9 1058.66     352  1058.9
   391.1 1059.38     4231059.025     4451059.015   459.6 1059.28   469.4 1060.04
   518.2 1064.94     528 1066.05   537.8 1067.52   576.9 1074.74   664.9 1091.78
   723.6 1103.92   762.7 1112.54   772.5  1114.5   782.2 1116.32   811.6 1121.18
#Mann= 3 , 0 , 0
       0     .06       0     423    .045       0     445     .08       0
Bank Sta=423,445
XS Rating Curve= 0 ,0
Exp/Cntr=0.3,0.1

Type RM Length L Ch R = 1 ,29148.6 ,513.4,513.5,513.4
XS GIS Cut Line= 2
     1684687.872      747057.988     1683923.983      747064.933
#Sta/Elev= 30
       0 1092.72    19.6 1087.42    29.4 1084.56    39.2 1081.13      49 1078.19
    58.8 1077.32    68.6 1077.14    78.4  1075.9   137.1  1061.7   146.9 1059.93
   156.7 1058.95   166.5  1058.8   225.3 1058.87     284  1060.1   313.4 1059.01
     333 1058.27   342.8 1058.42   363.6 1060.31     382 1062.21   391.8 1063.03
   460.3  1066.9   470.1 1067.77   479.9 1068.91   519.1  1073.8   636.6 1090.93
   695.4 1100.12   705.2 1101.76   724.8 1105.42   744.3 1108.71   763.9  1111.4
#Mann= 3 , 0 , 0
       0     .06       0   313.4    .045       0   363.6      .1       0
Bank Sta=313.4,363.6
XS Rating Curve= 0 ,0
Exp/Cntr=0.3,0.1

Type RM Length L Ch R = 1 ,28635.1 ,497.3,498,498.1
XS GIS Cut Line= 2
     1684803.324       746552.78     1683998.636      746557.988
#Sta/Elev= 30
       0  1118.3    19.6  1113.1    39.2 1108.23     157 1079.87   166.8 1077.89
   176.6 1076.87   186.5  1076.5   196.3 1075.57   206.1 1073.32   255.2 1058.61
     265 1056.07   274.8 1054.64   284.6 1054.42   333.7 1055.16   402.4 1055.06
   451.4 1055.59   490.7 1055.63   529.9 1055.74   549.6 1056.04   559.4 1057.36
   588.8 1065.26   608.4 1070.92   628.1 1077.07   647.7 1083.77   657.5 1086.81
   667.3 1089.23   677.1 1090.86   706.6 1093.91   755.6 1102.56   804.7 1112.29
#Mann= 3 , 0 , 0
       0     .08       0   490.7    .045       0   529.9      .1       0
Bank Sta=490.7,529.9
XS Rating Curve= 0 ,0
Exp/Cntr=0.3,0.1

Type RM Length L Ch R = 1 ,28137.1 ,282.9,296,308.8
XS GIS Cut Line= 3
     1684685.865      746110.122     1684586.906      746076.268
     1684081.698       746071.06
#Sta/Elev= 30
       0 1071.69     9.5 1069.61      19 1067.74    28.5 1066.52    47.5 1065.81
      57 1064.91    66.6 1063.53    85.6 1060.46    95.1 1059.01   114.3 1056.28
     124 1055.14   133.7 1054.32   143.4 1053.93   162.9 1053.71   211.5  1054.1
   269.8 1054.16   396.1    1053     4001053.056   405.8 1053.14   415.5 1053.54
     4251054.225   434.9    1056   444.6 1059.73   473.8 1074.26   493.2 1083.79
     503 1088.72   512.7 1093.77   522.4 1097.34   532.1 1099.12   609.8 1111.03
#Mann= 3 , 0 , 0
       0     .07       0     400    .045       0     425     .08       0
Bank Sta=400,425
XS Rating Curve= 0 ,0
Exp/Cntr=0.3,0.1

Type RM Length L Ch R = 1 ,27841.1 ,87.8,87.7,87.6
XS GIS Cut Line= 4
     1684733.011      746073.613     1684261.657      745761.113
     1684196.553      745813.196     1683865.824      745925.176
#Sta/Elev= 30
       0 1080.38    68.2 1066.19      78 1064.47    87.8  1063.4   107.3 1062.32
     117 1061.44   146.3 1057.55     156 1056.52   175.5 1055.12     195 1054.33
   224.3 1054.07     312 1054.85   419.3  1054.3   487.5 1052.57   502.71051.913
   526.5 1049.66   536.3  1050.6     546 1053.11   565.5 1058.65   584.1 1062.23
   593.3 1064.62   639.6 1078.38   726.5  1098.9   755.6 1106.97   765.3 1109.28
   833.2 1120.62   862.3 1126.07   881.7 1130.47   930.2 1142.54   998.1 1158.53
#Mann= 3 , 0 , 0
       0      .1       0   502.7    .045       0     546      .1       0
#XS Ineff= 2 , 0
          331.03 1057.39
Permanent Ineff=
       F       F
Bank Sta=502.7,546
XS Rating Curve= 0 ,0
Exp/Cntr=0.3,0.1

Type RM Length L Ch R = 1 ,27753.4 ,135.8,105.5,74.7
XS GIS Cut Line= 4
     1684774.678      745998.092     1684303.324      745685.592
     1684217.386      745766.321     1683886.657      745878.301
#Sta/Elev= 30
       0 1087.41    87.8 1068.58   126.8 1061.55   146.3 1059.81     195 1057.09
   253.5 1055.09   409.5 1054.62   487.5 1053.51   497.3 1053.13     507 1051.97
   516.8 1049.81   526.5  1048.5   536.3 1048.61     546 1050.16   555.8 1052.03
   565.5 1053.07     595  1055.1   614.7 1055.72   624.5 1057.34   644.1 1063.12
   673.6 1069.75   702.8 1078.48   741.6    1088   780.4 1100.36   790.1 1102.89
   819.2 1108.13   896.8 1118.99   925.9 1123.78   945.3 1127.86  1032.6 1148.79
#Mann= 3 , 0 , 0
       0      .1       0   516.8    .045       0     546      .1       0
Bank Sta=516.8,546
XS Rating Curve= 0 ,0
Exp/Cntr=0.3,0.1

Type RM Length L Ch R = 1 ,27647.9 ,820.6,825.5,828.5
XS GIS Cut Line= 4
     1684703.497      745015.453     1684660.094      745319.273
     1684156.622      745770.662     1683765.997      745883.509
#Sta/Elev= 30
       0  1105.7    67.1 1090.02     163 1074.51   201.4 1070.06   239.8 1068.75
     259 1067.16   326.5 1057.27   375.5 1049.05   434.3 1048.81   463.7 1050.37
   522.5 1050.96   649.9  1047.6   698.9  1047.4     7381047.459     7621048.366
   787.1 1050.03   845.9 1056.36   865.5 1057.35   875.3 1058.54   904.7 1069.56
   924.3 1075.86   983.1 1090.13  1002.5 1097.08  1021.8 1101.82  1060.5 1108.38
    1138  1118.6    1167 1123.13  1186.4 1127.08  1302.6 1154.37  1389.7 1169.39
#Mann= 3 , 0 , 0
       0      .1       0     738    .045       0     762      .1       0
#XS Ineff= 2 , 0
          531.03 1054.57
Permanent Ineff=
       F       F
Bank Sta=738,762
XS Rating Curve= 0 ,0
Exp/Cntr=0.3,0.1

Type RM Length L Ch R = 1 ,26822.4 ,345.2,345.5,345.5
XS GIS Cut Line= 2
     1684385.713      744718.332      1683614.88      745169.721
#Sta/Elev= 30
       0    1097   196.3 1050.72     216 1046.18   225.8 1044.44   235.6  1043.9
   264.31044.243   314.1 1046.71   353.4  1047.7   382.8 1047.67   441.7 1046.24
   471.2 1046.47   490.8 1047.53   510.4  1049.2   520.3 1050.32   549.7 1054.37
   559.5 1056.41   569.3 1059.95   598.8 1073.04   608.6 1076.59   618.4 1078.38
   628.2 1078.84     638 1079.83   647.9 1081.58   687.1 1090.09   755.8 1104.39
   775.5 1108.96   795.1 1114.49   814.7 1120.89   863.8 1137.79   893.3 1146.77
#Mann= 3 , 0 , 0
       0      .1       0   225.8    .045       0   264.3     .08       0
Bank Sta=225.8,264.3
XS Rating Curve= 0 ,0
Exp/Cntr=0.3,0.1

Type RM Length L Ch R = 1 ,26476.9 ,288.8,286.9,284.4
XS GIS Cut Line= 2
     1684101.494      744522.488     1683543.768      744834.988
#Sta/Elev= 30
       0 1070.82    19.7 1066.21    29.5  1063.5    68.8 1051.03    88.5  1045.6
    98.4 1044.14   108.2 1043.81     118  1043.8   127.9  1043.8   157.4 1043.83
   186.9 1044.27   216.4 1045.51   245.9 1044.66   295.1  1044.8   324.6 1045.95
   363.9  1048.2   383.6 1049.54   393.4 1050.67   403.3 1052.59   452.4 1063.96
   462.3 1065.62   472.1 1066.29   481.9  1066.6   491.8 1067.82   501.6 1070.41
   531.1 1079.05   560.6 1087.01   590.1 1094.57   609.8 1098.71   639.3 1103.95
#Mann= 3 , 0 , 0
       0      .1       0   108.2    .045       0   127.9     .08       0
Bank Sta=108.2,127.9
XS Rating Curve= 0 ,0
Exp/Cntr=0.3,0.1

Type RM Length L Ch R = 1 ,26190   ,532.6,532.8,531.1
XS GIS Cut Line= 4
     1683923.542      744272.922      1683884.48      744314.155
     1683493.855      744574.571     1683469.983      744778.564
#Sta/Elev= 30
       0 1077.48     9.5 1073.91    18.9 1069.94    47.3 1057.14    66.6 1049.21
    76.4  1045.5    86.1 1042.84    95.9  1042.5   105.7  1042.5   125.3 1042.97
   144.8 1044.47   154.6 1044.37   164.4 1043.66   174.2  1043.4     184 1043.46
   232.8 1045.27   262.2 1044.82   301.3 1046.19   399.1 1050.58   467.6 1056.47
   477.4  1057.1   496.9 1057.46   506.7 1058.05   526.3 1060.53   555.6 1064.93
   594.7 1071.36   614.3 1075.23   663.2 1086.06   692.5 1091.53   731.7 1099.83
#Mann= 3 , 0 , 0
       0      .1       0    86.1    .045       0   105.7     .08       0
Bank Sta=86.1,105.7
XS Rating Curve= 0 ,0
Exp/Cntr=0.3,0.1

Type RM Length L Ch R = 1 ,25657.3 ,485.7,462.6,437.9
XS GIS Cut Line= 4
     1684131.109      743785.147     1683639.254      743862.766
     1683150.973      744164.415     1683007.744      744374.919
#Sta/Elev= 30
       0 1146.08    78.1  1139.7    97.6 1137.52   244.1  1110.5   273.4 1104.23
   292.9 1099.18   341.7 1085.52   390.5 1069.41   410.1 1063.49   439.4 1055.87
   458.9 1051.96   478.4  1049.1   497.9 1046.81     566  1040.7   585.5 1039.63
   595.2  1039.6   605.2  1039.6     673 1039.64   721.7 1042.34   731.4 1042.45
     780 1040.68   789.8 1040.71   867.6 1043.97  1003.8 1044.23    1033 1044.98
  1071.9 1047.84  1189.4 1058.62  1277.5  1067.8  1306.9 1070.17  1326.5 1073.06
#Mann= 3 , 0 , 0
       0      .1       0   585.5    .045       0   605.2     .08       0
Bank Sta=585.5,605.2
XS Rating Curve= 0 ,0
Exp/Cntr=0.3,0.1

Type RM Length L Ch R = 1 ,25194.6 ,200.4,210.7,221.1
XS GIS Cut Line= 4
     1683172.776      743233.064     1683161.824      743717.367
     1683166.164      744060.249     1682986.042      744325.005
#Sta/Elev= 30
       0 1143.02    67.8 1130.18   145.3 1116.55   290.7 1093.17   348.8 1082.77
   368.2 1078.94   406.9 1070.64     465  1057.3   494.2 1050.87   513.8 1046.98
   553.5 1039.76   562.8 1039.03   582.4 1038.93   592.2  1038.9   641.2 1039.04
   709.8 1041.18   729.4 1042.06   758.8 1044.11   768.6 1044.51   778.4 1044.62
   807.7 1044.23     837 1044.41   866.2 1044.87   875.8 1045.16   895.3 1046.16
   924.4 1048.27   963.2 1051.63  1040.8  1059.3  1069.9 1062.59  1147.6 1072.54
#Mann= 3 , 0 , 0
       0      .1       0   553.5    .045       0   582.4     .08       0
Bank Sta=553.5,582.4
XS Rating Curve= 0 ,0
Exp/Cntr=0.3,0.1

Type RM Length L Ch R = 1 ,24983.9 ,279.9,280.6,280.6
XS GIS Cut Line= 4
     1683068.609      743490.008     1682981.702      743689.155
     1682812.431      744051.568     1682779.879        744238.2
#Sta/Elev= 30
       0 1086.96     9.4 1085.32    37.8 1079.85   103.9 1066.93   151.2 1057.82
     227 1042.89   236.8 1041.12   246.6 1039.61     256 1038.71   266.1 1038.38
   285.6 1038.47   324.6 1038.71   344.1 1038.69   392.9  1038.3   422.2 1038.31
   451.4 1038.46   480.7 1039.23     510 1040.22   529.5 1041.02   539.2 1041.51
   558.7 1042.67   578.2 1044.08   597.8 1045.83   617.3 1047.69   683.6 1055.19
     712  1058.3     731 1060.55   749.9 1063.17   778.3 1067.74   806.7 1072.53
#Mann= 3 , 0 , 0
       0      .1       0     256    .045       0   285.6      .1       0
Bank Sta=256,285.6
XS Rating Curve= 0 ,0
Exp/Cntr=0.3,0.1

Type RM Length L Ch R = 1 ,24703.3 ,416.4,405.8,391.5
XS GIS Cut Line= 4
      1682788.56      743552.436     1682708.265      743632.731
     1682562.865      743953.912     1682512.952      744209.988
#Sta/Elev= 30
       0 1065.62    18.9 1062.66    47.3 1057.96    56.8  1056.1    66.2 1053.96
    85.2 1048.66    94.6 1046.84   123.4 1041.86   154.2 1037.21   162.5 1036.38
   172.3 1036.24   191.9 1036.82   221.3 1037.59   250.7 1037.96   299.6 1038.94
   348.6 1039.65   387.8 1040.37   417.2  1041.2   446.5 1042.39   495.1 1045.14
   543.4 1047.45   582.1  1049.6   601.4 1050.92   620.7 1052.57   630.4 1053.64
     640 1054.94   688.4 1061.71     698 1063.36   707.7 1065.22     727 1069.48
#Mann= 3 , 0 , 0
       0      .1       0   154.2    .045       0   191.9      .1       0
Bank Sta=154.2,191.9
XS Rating Curve= 0 ,0
Exp/Cntr=0.3,0.1

Type RM Length L Ch R = 1 ,24297.5 ,185.2,195.5,203.5
XS GIS Cut Line= 4
     1682371.893      743519.884     1682354.532       743608.86
     1682350.192      743962.592     1682384.914      744190.457
#Sta/Elev= 30
       0 1056.99    27.2 1053.42    36.3 1052.12    63.5 1047.26    72.5 1045.76
    90.6 1043.08   110.3 1040.48   120.1 1039.34     130 1038.43   147.5 1037.19
   159.4 1036.54   169.3 1036.14   208.6 1034.88     238 1034.27   257.7  1034.2
   277.4 1034.28   316.7 1034.87   346.2 1035.43   375.6 1036.31   385.4 1036.72
   405.1 1037.79   444.4 1040.53   482.8 1043.75   550.1  1049.1   607.7 1053.11
   617.3 1053.86   636.5  1055.6   646.1 1056.66   655.7 1057.86   674.9 1060.75
#Mann= 3 , 0 , 0
       0      .1       0     130    .045       0   147.5      .1       0
Bank Sta=130,147.5
XS Rating Curve= 0 ,0
Exp/Cntr=0.3,0.1

Type RM Length L Ch R = 1 ,24102   ,450.9,439.9,421.6
XS GIS Cut Line= 4
     1682246.025      743480.821     1682224.324      743576.308
     1682061.563      743910.509     1682059.393      744131.863
#Sta/Elev= 30
       0 1059.79      49 1050.52    68.5 1047.15    97.9 1042.77   127.3  1038.2
     137 1036.81   138.8 1036.64   146.8 1035.91   156.6 1035.76   176.2 1035.38
   195.7 1034.48   205.5  1034.2     274 1034.31   322.9 1035.32     411 1037.56
   450.1 1038.93   469.6 1039.79   488.9 1040.47   517.8 1041.06   527.4 1041.14
     537 1040.72   546.6  1039.7   556.3  1038.2   565.9 1037.58   575.5 1037.66
   594.8 1038.67   623.6 1040.85   633.3  1041.8   671.8 1045.94     691  1047.8
#Mann= 3 , 0 , 0
       0      .1       0   138.8    .045       0   156.6      .1       0
Bank Sta=138.8,156.6
XS Rating Curve= 0 ,0
Exp/Cntr=0.3,0.1

Type RM Length L Ch R = 1 ,23662.1 ,486.1,482.1,440.9
XS GIS Cut Line= 4
     1681833.699      743380.995     1681827.188      743485.162
     1681944.376      743886.637     1681963.907      744175.266
#Sta/Elev= 30
       0 1053.67      38 1050.02    75.9 1045.92   143.3  1037.7   154.8 1035.91
   162.7 1034.91   172.4 1034.51   182.2 1034.69   201.6 1035.05   230.8 1035.01
   269.7 1033.65   289.2 1033.47   328.1  1033.8   357.2 1034.48   386.4 1035.67
   425.3  1037.7   454.5 1038.71     474 1038.93   493.4 1038.35   503.2 1038.52
   541.9 1041.26   561.2 1042.27   570.8  1042.6   590.1 1042.95   609.4 1043.15
   628.7 1043.13     648 1043.51   725.1 1045.77     783 1047.96   811.9 1049.36
#Mann= 3 , 0 , 0
       0      .1       0   154.8    .045       0   182.2      .1       0
Bank Sta=154.8,182.2
XS Rating Curve= 0 ,0
Exp/Cntr=0.3,0.1

Type RM Length L Ch R = 1 ,23180   ,299.5,318.2,338
XS GIS Cut Line= 3
     1681351.928      743480.821     1681473.456      743673.964
      1681851.06      744129.693
#Sta/Elev= 30
       0 1043.92      38 1043.41    66.6 1042.71    95.1  1041.8   161.6 1039.46
   228.2 1037.48     267 1035.97   315.5 1033.53   334.9 1032.65   344.6 1032.29
   359.6 1031.91   393.1 1031.38   412.5 1031.08   431.9 1030.64   441.6  1030.6
   470.8 1030.74   480.4 1031.14   499.9  1033.4   509.6 1034.12   519.3  1034.6
   548.4 1035.76   587.2 1037.08   674.5 1039.81     723 1041.03   742.4 1041.68
   752.1 1042.18   761.8 1042.92   781.2 1044.87   790.9 1045.62     820 1047.47
#Mann= 3 , 0 , 0
       0     .08       0   359.6    .045       0   393.1     .07       0
Bank Sta=359.6,393.1
XS Rating Curve= 0 ,0
Exp/Cntr=0.3,0.1

Type RM Length L Ch R = 1 ,22861.8 ,147.4,148.4,146.7
XS GIS Cut Line= 3
     1681323.716      743660.943     1681304.185       743771.62
     1681291.164      744292.453
#Sta/Elev= 30
       0 1040.97    28.1 1040.14    65.6 1039.42    74.9 1039.09    93.7 1038.16
   151.7 1034.18   171.4 1033.01   181.2 1032.54   220.5 1030.98   230.4  1030.7
   240.2 1030.24   246.6 1029.77     250 1029.52   259.8 1029.22   269.7 1029.66
   279.5 1030.45   289.3 1031.01   299.2 1031.06   318.8 1030.35   328.6 1030.15
   358.1 1030.21   387.6 1030.54   436.8 1031.35   456.4 1031.82   476.1 1032.42
   564.6  1036.1   603.9 1037.92   613.7 1038.97   623.6 1040.78   633.4 1042.97
#Mann= 3 , 0 , 0
       0     .06       0   246.6    .045       0   269.7     .07       0
Bank Sta=246.6,269.7
XS Rating Curve= 0 ,0
Exp/Cntr=0.3,0.1

Type RM Length L Ch R = 1 ,22713.5 ,54.3,54.5,54.3
XS GIS Cut Line= 2
     1681210.869      743604.519     1681202.188      744272.922
#Sta/Elev= 30
       0 1041.59    39.3 1039.72    98.3 1037.84   186.8  1034.2   255.6 1032.88
   314.6 1032.93   324.4 1032.71   344.1 1031.02   353.9 1030.67   373.6 1031.34
   383.4 1030.56   393.2 1029.26     403  1028.9   412.9 1030.34   422.7 1032.35
   432.5 1033.46   442.4  1033.9   452.2  1034.1     462 1034.01   491.5 1032.83
   511.2 1032.78   530.8 1033.37   560.3 1034.95   589.8 1036.21   619.3 1035.92
   629.1 1036.19     639 1036.77   648.8 1037.69   658.6 1039.04   668.5  1040.7
#Mann= 3 , 0 , 0
       0     .06       0   383.4    .045       0   412.9     .06       0
Bank Sta=383.4,412.9
XS Rating Curve= 0 ,0
Exp/Cntr=0.3,0.1

Type RM Length L Ch R = 1 ,22659   ,91.6,92.1,92.4
XS GIS Cut Line= 2
     1681156.615       743608.86     1681147.935      744277.262
#Sta/Elev= 30
       0 1040.84    29.5 1040.17      59 1038.15    78.6 1037.01   127.8 1034.41
   157.3 1033.08     177 1031.86   196.6 1030.35   206.4 1029.78   216.3 1029.48
   235.9 1029.34   265.4 1029.67   294.9 1031.29   304.7 1031.72   314.6  1031.9
   324.4 1031.68   344.1 1030.38   363.7 1030.17   373.6 1029.58   383.4 1028.68
   393.2 1028.87   400.6 1030.24   412.9 1032.63   422.7 1033.57   432.5 1033.69
   491.5 1032.94   511.2 1033.08     521 1033.51   619.3 1039.04   668.5 1042.09
#Mann= 3 , 0 , 0
       0     .06       0   363.7    .045       0   400.6     .06       0
Bank Sta=363.7,400.6
XS Rating Curve= 0 ,0
Exp/Cntr=0.3,0.1

Type RM Length L Ch R = 1 ,22566.8 ,290.8,287,278.9
XS GIS Cut Line= 4
     1681113.748      743542.092      1681071.98      743686.985
     1681052.449      744212.158     1681063.299      744377.089
#Sta/Elev= 30
       0  1046.2    37.7 1044.69    84.8 1042.28    94.2 1041.23   131.9    1035
   141.4  1033.7   150.8 1032.69   160.5 1031.94   189.7  1030.2   218.9  1029.1
   248.1 1028.52     287  1028.2   345.4 1028.13   374.6 1028.26   423.3 1029.14
     433 1029.09   442.8 1028.69   453.4  1028.3   462.2 1028.35     472 1028.76
   481.7  1029.9   491.4 1030.77   549.8 1030.59   588.7 1031.47   627.7  1032.9
   656.9 1034.58   715.2 1038.99     793 1043.43   812.4 1044.79   841.6 1047.29
#Mann= 3 , 0 , 0
       0     .06       0   442.8    .045       0     472     .06       0
Bank Sta=442.8,472
XS Rating Curve= 0 ,0
Exp/Cntr=0.3,0.1

Type RM Length L Ch R = 1 ,22279.9 ,548.4,545.1,540.7
XS GIS Cut Line= 4
     1680752.969      743637.071     1680772.501      743723.877
     1680839.775      744060.249     1680867.987      744364.068
#Sta/Elev= 30
       0 1047.33    17.8 1043.24    26.7 1041.45    44.5  1038.5    53.4 1037.18
    71.2  1035.1    80.1 1034.32    98.8 1033.15   108.6 1032.27   147.8 1027.89
   157.6 1027.37     187  1027.1   206.6 1027.16     236 1028.04   255.6 1028.15
   265.4 1027.44   274.2 1027.06     285 1026.96   289.2 1027.48   304.6 1029.56
   314.4 1030.34   324.2 1030.66     432 1032.25   527.4  1033.4   546.4 1033.88
   594.1 1035.79   622.7 1037.45   641.8 1039.01   670.4 1041.67   737.1 1048.56
#Mann= 3 , 0 , 0
       0     .06       0   255.6    .045       0   289.2     .06       0
Bank Sta=255.6,289.2
XS Rating Curve= 0 ,0
Exp/Cntr=0.3,0.1

Type RM Length L Ch R = 1 ,21734.8 ,560,561.1,560.4
XS GIS Cut Line= 2
      1680299.41      743756.429     1680579.358      744374.919
#Sta/Elev= 30
       0  1058.7    68.9 1047.06    78.7  1045.2    88.6 1042.02    98.4 1037.66
   108.2 1033.46   118.1 1029.68   127.9 1026.35   137.8 1024.22   145.1 1023.83
   147.6  1023.7   167.3  1023.7   226.3 1023.73   236.1 1023.95     246 1024.56
   265.7 1025.98   285.3  1027.2   324.7 1029.13   344.4 1029.72     364 1030.05
   373.9 1030.11   432.9 1030.11   462.4  1030.4     492 1031.07   521.5 1032.25
   531.3 1032.77   560.8 1034.71   580.5 1036.15   590.3  1037.1   678.9 1047.67
#Mann= 3 , 0 , 0
       0      .1       0   145.1    .045       0   167.3     .06       0
Bank Sta=145.1,167.3
XS Rating Curve= 0 ,0
Exp/Cntr=0.3,0.1

Type RM Length L Ch R = 1 ,21173.7 ,347.2,376,386.3
XS GIS Cut Line= 5
     1680047.674      743864.936     1680036.824      743962.592
     1680197.414      744272.922     1680327.622      744485.596
     1680547.776      744649.731
#Sta/Elev= 30
       0 1046.39    68.8 1037.13   127.4 1025.07   137.1 1023.85   146.8  1023.7
   156.5  1023.7   224.4 1023.81   253.6 1025.39   321.5 1026.82   331.2  1026.5
   350.6 1024.46   360.3 1024.15     370  1024.6   389.4 1028.35   408.8 1029.74
     438 1033.61   447.7 1033.42   457.3 1031.85   476.4 1025.62     486 1024.26
   562.8  1025.1   620.3 1027.35     697 1031.97   706.8 1032.95   726.5 1036.41
   795.1 1051.81   814.7 1055.31     903 1064.29     952 1069.76   971.6 1071.43
#Mann= 3 , 0 , 0
       0      .1       0   137.1    .045       0   156.5      .1       0
#XS Ineff= 2 , 0
                          438.44         1041.35
Permanent Ineff=
       F       F
Bank Sta=137.1,156.5
XS Rating Curve= 0 ,0
Exp/Cntr=0.3,0.1

Type RM Length L Ch R = 1 ,20797.7 ,296.8,296.9,296.6
XS GIS Cut Line= 3
     1679887.084      743906.169     1679893.594      744014.676
     1679867.553      744680.908
#Sta/Elev= 30
       0 1038.51    45.3    1033    90.6 1027.98   108.7 1026.52   138.1 1024.86
   177.3  1022.3   206.8 1020.04   216.6 1019.37   226.4 1019.19   236.2 1019.65
   238.7 1020.15   255.8 1023.56   265.6 1024.68   275.4 1024.82   285.2 1023.84
     295 1022.49   304.8 1021.68   353.8 1021.21   383.2 1021.13   402.8 1021.24
   412.7 1021.38   422.5 1021.78   442.1 1022.95   451.9 1023.36   491.1 1024.36
     599 1025.73   657.8 1026.08   687.2 1026.43   706.8  1026.8   775.4 1029.19
#Mann= 3 , 0 , 0
       0     .06       0   206.8    .045       0   238.7     .06       0
Bank Sta=206.8,238.7
XS Rating Curve= 0 ,0
Exp/Cntr=0.3,0.1

Type RM Length L Ch R = 1 ,20500.7 ,350.2,355.2,350.6
XS GIS Cut Line= 4
     1679644.028      743888.808     1679633.178      743951.742
     1679620.157      744459.554     1679561.563      744641.846
#Sta/Elev= 30
       0 1033.66    36.5 1029.52    63.9 1026.21    73.6  1025.3    83.4 1024.75
   102.9 1024.13   161.6 1022.91   190.9 1022.11   259.2 1019.05   278.8 1018.38
   288.6 1018.22   308.1 1018.16   317.8 1018.15   327.6 1018.17   347.2 1018.26
   356.9 1018.49   386.2 1019.75   464.4 1023.63     523 1026.13   581.4 1027.92
   600.6  1028.6   610.1 1029.07   619.7 1030.18   629.3 1031.97   638.9 1034.07
   686.7 1045.04     725  1053.6   734.6 1055.38   744.2 1056.66   763.3 1058.68
#Mann= 3 , 0 , 0
       0     .07       0   308.1    .045       0   327.6     .06       0
Bank Sta=308.1,327.6
XS Rating Curve= 0 ,0
Exp/Cntr=0.3,0.1

Type RM Length L Ch R = 1 ,20145.5 ,328.1,321.6,276.8
XS GIS Cut Line= 4
     1679489.949      743880.127     1679444.376      743962.592
      1679353.23      744296.794     1679322.848      744528.999
#Sta/Elev= 30
       0 1030.52     9.4 1030.28    37.7 1030.32    47.1 1030.17    56.5  1029.9
    75.4 1028.76    94.2 1027.08   113.5 1024.82   123.1 1023.43   152.2 1018.63
   161.6 1017.77   171.2 1017.62   200.1 1017.66   238.6 1018.02   248.2 1018.32
   286.7  1020.7   296.3 1021.09   363.6 1021.92   392.5 1022.45   450.4 1024.16
   479.7 1025.39   489.4    1026   499.2 1026.99   538.2 1033.05   557.7 1035.27
   577.2 1036.92   616.3 1039.53   635.8 1041.33   655.3 1043.78   674.8 1046.99
#Mann= 3 , 0 , 0
       0     .07       0   152.2    .045       0   171.2     .06       0
Bank Sta=152.2,171.2
XS Rating Curve= 0 ,0
Exp/Cntr=0.3,0.1

Type RM Length L Ch R = 1 ,19824   ,798.7,789.3,737.3
XS GIS Cut Line= 4
     1679162.258      743743.408     1679166.598      743858.426
     1679183.959      744316.325     1679214.341      744515.978
#Sta/Elev= 30
       0 1034.76    57.6 1030.18    86.3 1027.54   115.1 1024.62   134.6 1022.45
   154.1 1020.15   172.8 1017.69   183.4 1016.69   187.8 1016.49   193.1 1016.24
   202.8 1016.07   222.3    1016   241.8 1016.08   271.1 1017.18   300.3 1018.08
   388.1 1020.54   436.8 1021.75   563.6 1023.77   582.9 1024.36   602.2 1025.37
     631 1027.43   650.3 1029.08   659.9 1030.02   688.7 1033.35   698.3 1034.75
     708 1036.63   727.2 1040.86   746.4 1044.82     756 1046.48   775.3 1049.19
#Mann= 3 , 0 , 0
       0      .1       0   172.8    .045       0   187.8     .06       0
Bank Sta=172.8,187.8
XS Rating Curve= 0 ,0
Exp/Cntr=0.3,0.1

Type RM Length L Ch R = 1 ,19034.7 ,247.4,258.9,269.6
XS GIS Cut Line= 4
     1678671.806      743817.193      1678726.06      743945.231
     1678936.563      744348.877     1678962.605      744539.849
#Sta/Elev= 30
       0 1036.81    74.2 1029.56   139.1 1023.45   197.2 1017.57   206.9 1016.69
   216.6 1015.94   227.6 1015.63   235.9  1015.6   245.6  1015.6     265 1015.63
   284.4 1015.92   352.2 1017.16   400.6 1017.66   458.7 1018.99   507.1 1020.31
   526.5 1020.94   545.9 1021.67   574.9 1022.89   594.3 1023.79   603.9 1024.32
   623.2 1025.52   642.5 1026.84   652.1 1027.69   661.8 1028.67   671.4 1029.76
   690.7 1032.17   729.2 1037.37   748.5 1040.14   767.8  1043.1     787 1046.16
#Mann= 3 , 0 , 0
       0      .1       0   227.6    .045       0   245.6     .06       0
Bank Sta=227.6,245.6
XS Rating Curve= 0 ,0
Exp/Cntr=0.3,0.1

Type RM Length L Ch R = 1 ,18775.8 ,216,227.9,238.5
XS GIS Cut Line= 3
     1678522.067      743884.467     1678522.067      744437.853
     1678563.299      744624.485
#Sta/Elev= 30
       0 1029.57     9.7 1028.53    19.4 1027.62    29.1  1026.8    38.8 1026.16
    48.5 1025.74      68 1025.46    77.7 1025.14    87.4 1024.53   126.2 1021.47
   135.9 1020.54   145.6  1019.1   155.3 1017.34   164.8 1016.05   174.8 1015.63
   184.5  1015.6     398  1015.6   407.8 1015.63   417.5 1015.82   427.2 1016.26
   475.7 1019.17   504.8 1020.72   514.6 1021.36   553.4  1024.4   610.7 1029.55
     649 1033.14   658.5 1034.09   668.1 1035.21   687.2 1037.72   744.5 1045.66
#Mann= 3 , 0 , 0
       0     .08       0   164.8    .045       0   184.5     .08       0
Bank Sta=164.8,184.5
XS Rating Curve= 0 ,0
Exp/Cntr=0.3,0.1

Type RM Length L Ch R = 1 ,18547.9 ,955.1,996.3,974.8
XS GIS Cut Line= 4
     1678472.153      743830.214     1678383.178      743958.252
     1678127.101      744420.492     1678135.782      744594.103
#Sta/Elev= 30
       0 1036.68      39 1032.77    87.7 1028.45   146.2 1022.64   165.7  1020.8
   175.5 1020.03   204.8 1018.03   234.2 1016.33     244 1015.88   253.8 1015.65
   263.6  1015.6   302.7  1015.6   322.3  1015.6     381 1015.62   390.8 1015.91
   400.6 1016.47   410.4 1016.75   478.8 1017.38   508.2 1017.76   557.1 1018.51
   606.1 1019.58   625.6 1020.33   645.2 1021.77   664.8 1022.88   703.7 1024.57
   780.9  1027.6   809.9 1028.98   819.6 1029.49   838.9 1030.81   858.2 1032.53
#Mann= 3 , 0 , 0
       0     .08       0   302.7    .045       0   322.3     .08       0
Bank Sta=302.7,322.3
XS Rating Curve= 0 ,0
Exp/Cntr=0.3,0.1

Type RM Length L Ch R = 1 ,17551.6 ,140.3,124.3,121.4
XS GIS Cut Line= 5
     1678186.664      742597.647      1678143.79      743241.411
     1677805.921      743786.811     1677960.001      744468.235
     1678053.317      744726.481
#Sta/Elev= 30
       0  1122.6   117.3 1126.04   205.3 1129.96   312.8 1139.26   527.9 1133.68
   576.8  1135.3   625.6 1138.65   645.2 1138.42   684.1 1127.64   752.1 1102.63
   771.6 1097.35   820.2 1087.68   868.8 1080.66     966 1064.78  1014.6 1055.81
  1131.2 1041.18    1209 1033.96  1267.3 1029.91  1306.4 1021.12  1326.1 1018.13
  1385.2 1016.58  1424.5 1013.82  1444.2  1013.6  1477.9 1013.65  1493.4 1014.43
  1522.9 1017.32  1611.5 1016.94  1975.6 1019.47  2093.3 1026.24    2260 1037.88
#Mann= 3 , 0 , 0
       0     .08       0  1477.9    .045       0  1493.4     .08       0
Bank Sta=1477.9,1493.4
XS Rating Curve= 0 ,0
Exp/Cntr=0.3,0.1

Type RM Length L Ch R = 1 ,17427.3 ,230.5,259.8,256.9
XS GIS Cut Line= 5
     1677283.887      742538.619      1677257.62      743528.191
     1677688.733      743715.196     1677905.747      744526.828
      1677955.66      744789.415
#Sta/Elev= 30
       0 1165.47    58.8 1158.96   215.6 1138.75   284.2 1125.28   372.4 1109.76
   450.8 1093.51   548.9 1075.33   607.7 1075.06   715.5 1083.33   774.3 1085.78
   980.1 1084.92  1019.3 1078.06  1087.8 1070.63  1166.1 1057.26    1264 1042.34
    1313 1036.19  1401.1  1028.4  1440.3 1020.98  1498.9 1017.12  1635.7  1013.6
  1655.2  1013.6  1684.5  1013.6  1713.8 1013.75  1772.5 1017.25  1821.3 1015.92
  1889.7 1015.97  2309.5 1020.23  2376.4 1023.77  2538.6 1035.83  2567.3 1039.06
#Mann= 3 , 0 , 0
       0     .08       0  1655.2    .045       0  1684.5     .08       0
Bank Sta=1655.2,1684.5
XS Rating Curve= 0 ,0
Exp/Cntr=0.3,0.1

Type RM Length L Ch R = 1 ,17167.5 ,535.3,505.3,503.4
XS GIS Cut Line= 4
     1677371.893      743823.703     1677541.164       743921.36
       1677792.9       744559.38     1677849.324      744815.457
#Sta/Elev= 30
       0 1052.12    19.5 1049.19    48.9 1045.23    87.9 1038.22   117.2  1032.6
   136.8 1029.31   175.9 1024.12   195.4 1021.79   205.2 1022.05     215  1021.1
   234.6 1016.34   244.4 1014.79   254.2 1013.99   303.2  1013.6   362.7 1013.72
   377.7 1014.37   401.2 1016.14     411 1016.56   499.2 1016.46   744.1 1018.49
   812.7 1019.19   861.7    1020   929.9 1020.58     959 1021.23   978.4 1022.02
   988.1 1022.72  1017.3 1025.78  1065.8 1029.75  1104.7 1033.75  1143.5 1038.15
#Mann= 3 , 0 , 0
       0     .08       0   362.7    .045       0   377.7     .08       0
Bank Sta=362.7,377.7
XS Rating Curve= 0 ,0
Exp/Cntr=0.3,0.1

Type RM Length L Ch R = 1 ,16662.2 ,494,495.1,492.4
XS GIS Cut Line= 3
     1677259.046      744016.846     1677269.896      744129.693
     1677499.931      744819.797
#Sta/Elev= 30
       0 1043.31    94.5 1031.06   103.9 1029.19   113.4 1025.85   123.2 1020.86
     133 1016.35   142.9 1013.76   152.7 1012.57   162.5  1011.9   172.4 1011.71
   182.2  1011.7     192 1011.72   211.7 1011.97   241.2 1012.68   300.1 1013.12
   398.4 1014.51   467.2 1015.85   506.6 1016.25   545.9 1016.26   575.4 1016.07
   604.9 1015.68     654 1014.78   663.9 1014.69   673.7 1014.84   703.2 1016.09
   732.7 1017.69   742.5 1018.42     772 1021.49   791.6 1023.71   840.8 1029.84
#Mann= 3 , 0 , 0
       0      .1       0     192    .045       0   211.7     .08       0
Bank Sta=192,211.7
XS Rating Curve= 0 ,0
Exp/Cntr=0.3,0.1

Type RM Length L Ch R = 1 ,16167.1 ,295.5,296.7,298.4
XS GIS Cut Line= 4
     1676957.396      744042.887     1676931.355       744240.37
     1677141.858      744843.669     1677211.303      745069.363
#Sta/Elev= 30
       0 1041.32    94.8 1033.67   151.8 1031.58   180.2 1029.78   189.7 1028.64
   199.2  1025.2   218.8 1014.73   228.7 1011.71   238.5 1010.22   258.2 1009.51
     268 1009.61   277.8 1010.04   307.3 1012.76   366.3 1014.81     386 1014.89
     445 1013.83   533.4  1013.1   641.6 1015.09     730    1016   798.8  1017.4
   808.7 1017.82   828.3  1019.4   887.4 1025.58   916.9 1029.49   946.4 1035.64
   956.2 1036.72   966.1 1037.19  1015.3 1037.68  1064.5 1037.63  1074.3 1038.32
#Mann= 3 , 0 , 0
       0      .1       0   238.5    .045       0     268     .06       0
Bank Sta=238.5,268
XS Rating Curve= 0 ,0
Exp/Cntr=0.3,0.1

Type RM Length L Ch R = 1 ,15870.4 ,447.1,448.4,446.5
XS GIS Cut Line= 4
     1676695.678      744167.887     1676733.872      744463.026
     1676912.692      744999.485     1676930.053      745159.207
#Sta/Elev= 30
       0 1034.45    57.6  1031.2      96 1028.56   163.2 1024.95   220.8 1024.35
   249.6 1023.44   268.8 1022.43     288 1020.59   297.6 1018.87   307.4 1015.85
   319.2  1011.5   326.8 1009.26   336.6 1008.21   356.1  1008.9   385.4 1009.87
   443.8 1009.81   482.8  1010.8   502.3 1010.73   512.1 1011.49   521.8  1011.8
   599.8 1013.32   648.6 1015.57   726.6 1015.92   833.8 1017.95   900.9 1020.13
   938.7 1020.62   957.6 1021.59   976.5 1022.11  1004.8 1025.67  1023.7 1025.42
#Mann= 3 , 0 , 0
       0      .1       0   319.2    .045       0   356.1     .08       0
Bank Sta=319.2,356.1
XS Rating Curve= 0 ,0
Exp/Cntr=0.3,0.1

Type RM Length L Ch R = 1 ,15422   ,204,203.9,204.5
XS GIS Cut Line= 4
     1676310.695      744441.325     1676355.834      744573.269
      1676505.14      744937.853     1676572.848      745177.436
#Sta/Elev= 30
       0 1028.13    27.9 1025.16    46.5 1023.44      93  1019.6   139.4 1016.12
   149.1 1014.88   158.7 1013.03   177.9 1008.52   187.6 1007.16   197.1  1006.9
   216.3  1006.9   225.9    1007   235.5 1007.51     274 1010.43   312.4 1012.14
   360.5  1013.3   446.9 1013.55   485.4 1014.15   523.8 1015.52   562.2 1017.23
   600.4 1019.29   648.3 1022.23   657.9 1022.54   686.6 1022.75   696.2 1023.11
   734.5 1025.34   744.1 1026.13   753.7 1027.16   763.2 1028.51   782.4 1031.86
#Mann= 3 , 0 , 0
       0      .1       0   187.6    .045       0   216.3     .08       0
Bank Sta=187.6,216.3
XS Rating Curve= 0 ,0
Exp/Cntr=0.3,0.1

Type RM Length L Ch R = 1 ,15218.1 ,179.9,180.9,181.4
XS GIS Cut Line= 4
     1676156.181      744592.367     1676206.528      744670.492
     1676324.584      745045.492      1676388.82      745252.089
#Sta/Elev= 30
       0 1022.26    37.2 1019.26    65.1 1017.24    92.9 1015.58   122.4 1014.17
   142.1 1012.94   151.9 1012.15   161.7 1010.39   171.6 1007.99   181.4 1006.85
   191.2  1006.8   210.9 1006.99   240.4 1008.82     260 1009.75     378 1011.14
   407.5 1011.77   476.3 1015.02   505.8 1017.27   525.4 1018.94   535.3 1019.94
   545.1 1021.21   554.9 1023.02   564.8 1025.89   574.6 1029.62   584.4 1032.33
   594.3 1033.15   633.6 1033.81   672.9 1034.09   682.8 1034.45   702.4 1036.32
#Mann= 3 , 0 , 0
       0     .06       0   171.6    .045       0   191.2     .06       0
Bank Sta=171.6,191.2
XS Rating Curve= 0 ,0
Exp/Cntr=0.3,0.1

Type RM Length L Ch R = 1 ,15037.2 ,146.8,151,156.6
XS GIS Cut Line= 4
     1676065.903      744611.464     1676046.806        744738.2
     1676145.765      745102.783     1676180.487       745278.13
#Sta/Elev= 30
       0 1023.86    91.6  1019.5   128.2 1017.43   137.8 1016.17   157.2 1011.28
   166.9 1009.78   176.6 1009.04   215.4 1006.62     225 1006.13   234.7    1006
   244.6 1006.42   292.8 1010.17   312.2 1011.23   331.6 1012.05     351 1012.66
   370.3 1013.03   428.4  1013.3   447.8 1013.54   467.2 1014.05   496.3 1015.42
   515.4 1016.79   534.2 1018.51     553 1020.68   590.6  1025.7   609.4 1027.73
   628.2 1029.38   637.6 1029.99   656.5 1030.68   665.9 1031.35   684.7 1033.25
#Mann= 3 , 0 , 0
       0      .1       0   215.4    .045       0   244.6     .07       0
Bank Sta=215.4,244.6
XS Rating Curve= 0 ,0
Exp/Cntr=0.3,0.1

Type RM Length L Ch R = 1 ,14886.1 ,312.7,308.2,301.2
XS GIS Cut Line= 4
     1675930.487      744635.769     1675927.015      744719.103
     1675930.487      745173.964     1675963.473      745325.005
#Sta/Elev= 30
       0 1021.23    83.4 1015.64    93.1 1014.83   102.8 1013.34   122.1 1008.75
   131.8 1007.03   141.5 1005.86   151.2 1005.15   160.8 1004.91   170.5  1004.9
   186.8  1004.9   209.2  1004.9   247.9 1004.97   257.6 1005.28   286.6 1007.07
   325.4 1009.13   364.1 1010.62   431.8 1012.11   470.5 1012.35   499.6 1013.28
   528.6 1014.99   567.3 1018.26   586.6  1020.5   625.2 1025.57   634.9 1026.63
   644.6 1027.31   663.9 1027.79   673.6 1028.23   683.2 1028.84   692.9 1029.74
#Mann= 3 , 0 , 0
       0      .1       0   186.8    .045       0   209.2     .06       0
Bank Sta=186.8,209.2
XS Rating Curve= 0 ,0
Exp/Cntr=0.3,0.1

Type RM Length L Ch R = 1 ,14577.9 ,115.7,115.3,114.8
XS GIS Cut Line= 4
     1675659.653       744581.95     1675656.181      744722.575
     1675808.959      745156.603     1675836.737      745349.311
#Sta/Elev= 30
       0 1023.95    65.6    1019    93.8 1017.11     170 1012.82   189.6 1012.01
   199.4  1011.8   209.2 1011.14     219 1008.82   222.4 1007.73   228.8 1005.67
   237.4 1004.69   238.6 1004.55   248.4 1004.69   287.5 1005.82   316.9 1006.07
     356 1006.14   424.6 1007.21   434.4 1007.83     454 1009.41   463.7 1009.88
   542.1 1012.94   581.2  1014.7   610.5  1016.3   649.5 1018.65   688.4  1021.3
   727.4 1024.34   737.1 1024.95   756.6  1025.9   766.3 1027.24   795.5 1032.99
#Mann= 3 , 0 , 0
       0      .1       0   222.4    .045       0   237.4     .07       0
Bank Sta=222.4,237.4
XS Rating Curve= 0 ,0
Exp/Cntr=0.3,0.1

Type RM Length L Ch R = 1 ,14462.6 ,265.7,256.8,247.4
XS GIS Cut Line= 4
     1675428.751      744614.936      1675536.39      744693.061
     1675704.792      745191.325     1675742.987      745366.672
#Sta/Elev= 30
       0 1029.43    28.5 1027.31    66.5 1025.24    85.5 1023.82   104.5 1021.57
   152.5 1014.01     172 1011.85   201.2 1010.15   249.9 1008.47   269.4 1006.68
   282.7 1004.91   288.8 1004.19   308.3 1003.76   327.8 1003.98     357 1003.66
   405.7 1002.14   415.5  1002.2   425.2 1002.74   434.9 1003.57   454.4 1006.31
   464.2 1006.99   600.5  1013.2     659  1015.6   715.6  1019.5   734.5 1021.34
   772.3  1025.7   791.2 1026.58   800.6  1027.6   810.1 1029.74   838.4 1037.86
#Mann= 3 , 0 , 0
       0      .1       0   282.7    .045       0   308.3     .08       0
Bank Sta=282.7,308.3
XS Rating Curve= 0 ,0
Exp/Cntr=0.3,0.1

Type RM Length L Ch R = 1 ,14205.8 ,401.3,411.5,420.7
XS GIS Cut Line= 4
     1675225.626      744845.839     1675312.431      744878.825
     1675626.667      745227.783     1675668.334      745382.297
#Sta/Elev= 30
       0 1028.43    46.4 1024.16    55.7 1022.81    83.6 1017.29    92.9 1015.76
   102.6 1014.53     132 1011.49   171.1 1007.92   180.9 1006.54   184.6  1005.8
   190.7 1004.57   199.6 1003.83   210.3 1003.73     220 1003.93   278.7 1006.85
     357 1008.22   396.1 1009.84   454.8 1011.41   523.3  1013.7   552.7 1015.06
   562.4  1015.8   628.4 1022.58   647.2 1024.69   656.6 1025.55     666 1026.02
   675.4  1026.8   684.8 1029.05   703.7    1036   713.1 1038.85   722.5  1040.2
#Mann= 3 , 0 , 0
       0     .06       0   184.6    .045       0   210.3     .08       0
Bank Sta=184.6,210.3
XS Rating Curve= 0 ,0
Exp/Cntr=0.3,0.1

Type RM Length L Ch R = 1 ,13794.4 ,109.3,110.1,111.2
XS GIS Cut Line= 4
     1675194.376      745061.117     1675275.973      745123.617
     1675354.098      745323.269     1675390.556      745418.755
#Sta/Elev= 30
       0 1022.93    46.7 1022.13    65.4  1021.4    74.8 1020.59    84.1 1019.19
    93.4 1017.52   102.8 1015.57   122.3 1012.51     132 1011.25   141.8 1010.57
   161.2 1009.76   180.7 1009.04     210 1008.14   219.7 1006.96   227.4 1005.35
   229.5 1004.91   239.2  1003.8     249  1004.4   258.7 1005.62   268.4 1006.98
   278.2  1008.5   297.7 1011.81   317.2 1015.48     345 1021.07   354.3  1022.4
   372.9 1023.89   382.2 1025.68   400.8 1031.56   410.1 1033.97   419.4 1035.89
#Mann= 3 , 0 , 0
       0     .06       0   227.4    .045       0     249     .08       0
Bank Sta=227.4,249
XS Rating Curve= 0 ,0
Exp/Cntr=0.3,0.1

Type RM Length L Ch R = 1 ,13684.2 ,50.9,50.7,50.7
XS GIS Cut Line= 2
     1675152.709      745083.686     1675281.181       745456.95
#Sta/Elev= 30
       0 1023.04    28.9 1022.39    38.5 1022.08    48.1 1021.47    57.8 1020.07
    67.4 1018.16    86.6 1014.11    96.3  1012.3   105.9 1011.18   115.5 1010.69
   125.2 1010.44   182.9 1009.39   192.6 1008.98   202.2 1007.61   211.8 1005.26
   217.7 1004.28   221.4 1003.67   231.1 1003.88   232.7 1004.13   240.7 1005.39
   298.5 1016.96   308.1 1018.44   317.7 1019.07   327.4 1020.17     337 1023.18
   346.6 1026.64   356.2 1028.83   365.9  1030.1   385.1 1032.22   394.8 1033.42
#Mann= 3 , 0 , 0
       0     .07       0   217.7    .045       0   232.7     .09       0
Bank Sta=217.7,232.7
XS Rating Curve= 0 ,0
Exp/Cntr=0.3,0.1

Type RM Length L Ch R = 1 ,13633.6 ,109.7,116.9,123.8
XS GIS Cut Line= 2
      1675107.57      745107.992     1675236.042      745481.255
#Sta/Elev= 30
       0 1022.89    19.3 1021.97    28.9  1021.2    38.5 1019.83    48.1 1017.97
    57.8 1015.92    67.4    1014      77 1012.61    86.6 1011.82   105.9 1010.87
   125.2 1010.02   163.7 1008.74   173.3 1008.27   182.9 1007.21   202.2 1004.05
   211.8 1003.36   221.4 1003.93   226.5 1004.89   231.1 1005.75   269.6 1014.11
   279.2 1016.09   288.8 1017.52   298.5 1018.22   308.1 1019.49   317.7 1022.86
   327.4    1027     337 1029.59   356.2 1031.86   365.9 1033.22   394.8 1037.53
#Mann= 3 , 0 , 0
       0     .08       0   202.2    .045       0   226.5     .08       0
Bank Sta=202.2,226.5
XS Rating Curve= 0 ,0
Exp/Cntr=0.3,0.1
