HEC-RAS study SFTOMLINRN.prj: SFTOMLINRN

--- SFTOMLINRN.g01 (geometry) --- (continued)

Type RM Length L Ch R = 1 ,13516.7 ,141.8,143,144.1
XS GIS Cut Line= 4
     1675072.848      745107.992     1675065.903      745201.742
     1675069.376      745354.519     1675083.265      745446.533
#Sta/Elev= 27
       0 1023.07    18.8 1021.63    28.2  1020.5    37.6  1019.1      47 1017.58
    56.4 1015.84    65.8 1014.23    75.2 1013.05   132.2 1008.23   141.8 1007.13
   160.9  1004.4   167.9 1003.66   170.4 1003.39     180 1003.21   189.5 1003.34
   199.1 1004.13   208.6 1005.56   218.2 1007.13   227.7 1008.81   265.4 1015.98
     284 1019.32   293.4 1020.37   302.7 1020.72     312 1022.36   321.3 1026.21
   330.6 1030.25   339.9 1032.81
#Mann= 3 , 0 , 0
       0     .06       0   167.9    .045       0   189.5     .08       0
Bank Sta=167.9,189.5
XS Rating Curve= 0 ,0
Exp/Cntr=0.3,0.1

Type RM Length L Ch R = 1 ,13373.7 ,100,100.4,100.9
XS GIS Cut Line= 3
     1674953.056      745116.672     1674932.223        745175.7
     1674925.278      745436.117
#Sta/Elev= 25
       0 1018.51    44.7 1012.04    53.6 1011.05    81.9 1008.29   120.5 1004.66
     126  1004.2   130.1 1003.86   139.8 1003.44   149.4 1003.36   159.1 1003.29
   178.4 1002.78     188 1002.68   197.7  1002.9   207.3 1003.36     217 1003.99
   226.6  1004.9   236.3 1006.32   245.9 1008.32   255.6 1010.75   274.9    1016
   284.5 1018.47   294.2 1020.73   303.8 1022.61   313.5 1023.64   323.1 1024.27
#Mann= 3 , 0 , 0
       0     .06       0     126    .045       0   149.4     .06       0
Bank Sta=126,149.4
XS Rating Curve= 0 ,0
Exp/Cntr=0.3,0.1

Type RM Length L Ch R = 1 ,13273.4 ,41.6,41.4,41.6
XS GIS Cut Line= 6
      1674763.82      745048.964     1674805.487       745121.88
     1674821.112      745172.228     1674833.265      745213.894
     1674828.056      745337.158      1674795.07      745462.158
#Sta/Elev= 30
       0 1017.01     9.3 1016.82    18.7 1016.31      56 1012.78    74.6 1011.22
   101.6 1009.45   136.7 1007.45   154.1 1006.73   162.7  1006.6   180.1 1006.92
   189.6  1006.7   199.1 1005.73   208.6 1004.04   218.1 1002.35   227.6 1001.89
     237 1002.76   246.5 1003.85     256 1004.25     275 1003.64   284.5 1003.59
     294 1004.01   303.5 1004.79   321.9 1006.86   331.2 1008.14   349.6 1011.03
   395.8 1016.65     405 1017.58   414.3 1018.08   423.5 1018.13   432.8 1018.75
#Mann= 3 , 0 , 0
       0     .06       0   208.6    .045       0   246.5     .06       0
Bank Sta=208.6,246.5
XS Rating Curve= 0 ,0
Exp/Cntr=0.3,0.1

Type RM Length L Ch R = 1 ,13232   ,248.1,259.7,270.3
XS GIS Cut Line= 6
      1674723.89      745043.755     1674765.556      745116.672
     1674781.181      745167.019     1674793.334      745208.686
     1674788.126       745331.95      1674755.14       745456.95
#Sta/Elev= 30
       0 1015.93     9.3 1014.98      28 1012.86    37.3 1012.17      56 1011.12
    74.6 1009.63    92.8 1008.36   127.9 1006.26   154.1 1004.93   162.7 1004.57
   171.4 1004.33   180.1 1004.26   199.1  1003.7   208.6 1003.23   218.1 1002.24
   227.6 1000.91     237 1000.55     249 1001.73     256  1002.5   265.5 1002.98
     294 1003.35   303.5 1003.73   312.7 1004.32   340.4 1006.81   349.6 1007.77
   377.4 1011.34     405 1015.19   414.3 1016.24   423.5 1016.84   432.8 1017.03
#Mann= 3 , 0 , 0
       0      .1       0   218.1    .045       0     249      .1       0
Bank Sta=218.1,249
XS Rating Curve= 0 ,0
Exp/Cntr=0.3,0.1

Type RM Length L Ch R = 1 ,12972.3 ,322.3,329.4,335.4
XS GIS Cut Line= 4
     1674708.265      745054.172     1674687.431       745090.63
     1674531.181      745357.992     1674487.778      745443.061
#Sta/Elev= 26
       0 1013.61      42  1007.4    51.7 1006.02    61.4 1004.83      71 1004.09
   109.7 1001.84   129.1 1001.25   138.8 1001.13   158.1 1001.29   177.5 1001.66
   187.2  1001.6   235.5 1000.69   264.6  999.95   274.2  999.86   293.6  999.82
   299.4 1000.05   303.3  1000.2     313 1001.53   332.3 1004.45   351.7 1007.71
   399.4 1016.62     409 1018.31   418.5 1019.89   428.1 1021.33   437.6 1022.66
   447.2 1023.88
#Mann= 3 , 0 , 0
       0      .1       0   274.2    .045       0   299.4      .1       0
Bank Sta=274.2,299.4
XS Rating Curve= 0 ,0
Exp/Cntr=0.3,0.1

Type RM Length L Ch R = 1 ,12642.9 ,305.9,294.8,263
XS GIS Cut Line= 4
     1674644.028      744908.339     1674512.084      744981.255
     1674328.056      745147.922     1674253.403      745297.228
#Sta/Elev= 30
       0 1027.34     9.4 1025.82    37.7 1020.52    47.1 1018.68      66  1014.8
   103.6 1006.81   113.1 1005.45   122.5 1004.69   160.3 1003.06   179.4 1001.99
     208  999.66   217.6  999.19   274.9  997.55     294  997.35   313.1  997.32
   332.2  997.38   340.4  997.73   341.7  997.79   370.4 1000.88   379.9 1001.81
     399  1003.5   448.1 1008.34     458 1008.97   477.6 1009.28   487.4 1010.32
   516.9 1015.07   536.5 1017.96   546.3 1019.33   556.1 1020.58     566 1021.64
#Mann= 3 , 0 , 0
       0     .08       0   313.1    .045       0   340.4     .08       0
Bank Sta=313.1,340.4
XS Rating Curve= 0 ,0
Exp/Cntr=0.3,0.1

Type RM Length L Ch R = 1 ,12348.1 ,1380.2,1355.4,1347.4
XS GIS Cut Line= 5
     1674445.345       744147.85     1674440.869      744563.843
     1674312.431      744765.978     1674177.015      745078.478
     1674173.542      745283.339
#Sta/Elev= 30
       0 1154.18    38.7 1141.31    67.7 1133.46    87.1 1129.62   135.4 1121.49
   212.8 1109.99   222.5    1109   309.6 1103.92   319.3 1102.24   348.3  1094.5
   377.3 1083.41     387 1080.46     416 1074.96   492.6 1058.75   569.3 1043.52
   588.4 1037.37   684.7 1001.18   694.4  998.54   704.2  997.35   723.6  996.79
   762.5  996.78   830.7  996.73     889  997.38   947.4 1001.32  1064.4 1007.47
  1083.9 1009.43  1113.2 1013.56  1171.7 1025.99  1181.5 1026.86    1201  1026.4
#Mann= 3 , 0 , 0
       0      .1       0   723.6    .045       0   762.5     .09       0
Bank Sta=723.6,762.5
XS Rating Curve= 0 ,0
Exp/Cntr=0.3,0.1

Type RM Length L Ch R = 1 ,10992.6 ,506.9,503,357.9
XS GIS Cut Line= 4
     1673303.852      744688.214     1673663.126      744866.672
     1673906.181       745153.13     1673975.626      745326.742
#Sta/Elev= 30
       0 1144.84   107.6 1097.92   166.3  1074.1   215.2 1054.89     225 1051.36
   254.4 1042.31   293.5 1029.35   332.7 1019.82   342.4 1016.15     362 1005.36
   371.8 1002.92     430  998.05     459   996.2   507.1  995.53   564.9   996.2
   593.8  996.12   632.3  995.17   670.9  993.14   690.1  992.91     703  993.11
   709.4  993.49   738.3   997.6   747.9  998.67   757.6   999.4   786.7 1000.05
   806.4 1002.11   835.9 1006.35   894.9 1016.26   934.3 1021.65   963.8 1025.03
#Mann= 3 , 0 , 0
       0      .1       0   670.9    .045       0     703     .09       0
Bank Sta=670.9,703
XS Rating Curve= 0 ,0
Exp/Cntr=0.3,0.1

Type RM Length L Ch R = 1 ,10489.6 ,235,241.6,374.2
XS GIS Cut Line= 4
     1673444.376      745094.103     1673498.195      745168.755
     1673682.223      745333.686     1673767.292      745390.978
#Sta/Elev= 30
       0 1022.13    18.4 1018.24    27.6 1015.82    55.2 1006.32    64.4 1003.35
    73.6 1000.93    82.8   999.1      92  997.45   101.5  995.46   120.9  990.91
     130   989.3   139.6  988.86   177.6  989.69   196.6  990.27   206.1  990.83
   225.1   992.4   234.6  992.98   253.6  993.81   263.1  994.12   272.6  994.18
   291.6  994.04   301.1  994.22   310.6  994.75   320.1  995.95   329.6  997.96
   367.1    1008   376.4 1010.06   385.8 1011.38   413.7 1014.64   441.7 1018.22
#Mann= 3 , 0 , 0
       0      .1       0   120.9    .045       0   139.6      .1       0
Bank Sta=120.9,139.6
XS Rating Curve= 0 ,0
Exp/Cntr=0.3,0.1

Type RM Length L Ch R = 1 ,10248   ,114.5,121.9,131.4
XS GIS Cut Line= 4
     1673314.167      745250.353     1673366.251      745342.367
     1673541.598      745578.478     1673650.973      745630.561
#Sta/Elev= 30
       0 1019.82    38.4 1013.91    57.7 1011.27    76.9 1008.82    86.5 1006.92
    96.1 1002.99   105.7  997.28   115.5  992.24   125.3  989.82   135.1  988.81
   165.6  986.47   174.4  986.11     194  986.05   213.6  986.33   233.2  987.11
     243  987.66   282.2  990.26   331.2  992.26     390  994.86   409.2  995.96
   418.5  996.71   427.8   997.8   437.1  999.63   455.7 1004.11   465.1 1006.53
   474.4 1009.14     493 1013.51   502.3 1015.34   511.7 1016.61     521 1017.61
#Mann= 3 , 0 , 0
       0      .1       0   165.6    .045       0     194      .1       0
Bank Sta=165.6,194
XS Rating Curve= 0 ,0
Exp/Cntr=0.3,0.1

Type RM Length L Ch R = 1 ,10126.1 ,67.2,74.7,80.1
XS GIS Cut Line= 4
     1673277.709      745330.214     1673300.278      745401.394
     1673364.515      745667.019     1673400.973      745779.867
#Sta/Elev= 30
       0 1012.57    18.7 1010.75    37.3 1009.18    46.7 1008.53    65.3 1007.74
    74.7 1004.05    84.4  996.54    94.2  990.86     104  988.76   113.7  987.99
   123.5   987.4   147.2  986.16   162.5  985.64   172.3   985.7   191.8  986.54
   221.1  988.22   250.4  990.59   260.1   991.1   269.9  991.39   289.4  991.59
   328.4   991.5   338.2   991.6     348  991.87   366.2  992.66   384.4  993.81
   402.7  995.25   430.1  997.66   439.2  998.99   448.3 1000.98   466.6 1005.52
#Mann= 3 , 0 , 0
       0      .1       0   147.2    .045       0   172.3      .1       0
Bank Sta=147.2,172.3
XS Rating Curve= 0 ,0
Exp/Cntr=0.3,0.1

Type RM Length L Ch R = 1 ,10051.4 ,43.4,41.5,41.5
XS GIS Cut Line= 2
     1673262.084      745321.533     1673253.403      745795.492
#Sta/Elev= 30
       0 1013.75      29 1010.87    48.4 1009.31      58 1008.75    67.7 1008.83
    77.4 1008.63    87.1  1004.6    96.7  996.94   106.4  991.02   116.1  988.78
   125.8  987.99   164.5  985.55   183.8  985.11   193.5   985.1   203.2  985.14
   208.6  985.38   212.8  985.56   232.2  987.96   241.9  988.86   261.2  989.88
   309.6  990.96     358  990.68   367.6  990.95   377.3  991.93   396.6   994.4
   406.3  995.85     416  997.69   425.7  999.83     445 1004.72     474 1013.13
#Mann= 3 , 0 , 0
       0      .1       0   183.8    .045       0   208.6      .1       0
Bank Sta=183.8,208.6
XS Rating Curve= 0 ,0
Exp/Cntr=0.3,0.1

Type RM Length L Ch R = 1 ,10009.9 ,109.1,117.1,125.1
XS GIS Cut Line= 2
     1673222.153      745314.589     1673213.473      745788.547
#Sta/Elev= 30
       0 1014.46      29 1011.39    48.4 1009.71    67.7 1008.38    77.4 1006.94
    87.1 1003.59   106.4  992.56   116.1   989.5   125.8  988.33   154.8  986.54
   174.1  985.48   183.8  985.19   203.2   985.1   222.5  985.14   225.8  985.25
   232.2  985.46   241.9   986.2   261.2  987.99   270.9   988.7   328.9  991.24
     358  992.67   367.6  993.35   377.3  994.39     387  995.65   396.6  997.08
     416 1000.43   425.7 1002.37     445 1006.56   454.7 1008.86     474 1013.85
#Mann= 3 , 0 , 0
       0      .1       0   203.2    .045       0   225.8      .1       0
Bank Sta=203.2,225.8
XS Rating Curve= 0 ,0
Exp/Cntr=0.3,0.1

Type RM Length L Ch R = 1 ,9892.7  ,270,272.8,273.6
XS GIS Cut Line= 4
     1673185.695      745342.367     1673156.181       745394.45
     1673078.056      745595.839      1673045.07      745748.617
#Sta/Elev= 23
       0 1010.66     8.6 1009.79    25.7 1007.62    34.2  1005.6    42.8 1002.76
    69.7  992.84    79.5  989.56    89.3  987.82    99.1   987.2     109  986.91
   187.5  985.38   207.1  984.98     217  985.03   226.8  985.73   236.6  986.89
   256.2  989.47   275.9  992.23   305.2  996.49     354  1003.3   373.6 1006.29
   412.6 1011.89   422.4 1013.49   432.2 1015.63
#Mann= 3 , 0 , 0
       0     .07       0   187.5    .045       0   226.8      .1       0
Bank Sta=187.5,226.8
XS Rating Curve= 0 ,0
Exp/Cntr=0.3,0.1

Type RM Length L Ch R = 1 ,9620    ,250.8,251.7,254
XS GIS Cut Line= 4
     1672994.723      745205.214     1672958.265      745257.297
     1672808.959      745531.603     1672765.556      745682.644
#Sta/Elev= 30
       0 1023.37    36.3  1017.1    45.4 1015.32    54.5 1012.48    63.6  1007.6
    73.3  998.68    83.1  989.87    92.8   985.6   102.6  984.43   131.9  983.44
   141.6  983.25   151.4   983.2   170.9   983.2   200.2   983.2   229.5  983.21
   239.2  983.37   258.8  983.97   278.3  984.68   297.8  985.52   317.3  986.67
   336.8  988.17   356.4  989.98   366.1  991.08   385.7  993.66   415.2   997.9
   444.6 1001.72   464.3 1003.94   503.6 1008.01   523.2 1010.27     533 1011.57
#Mann= 3 , 0 , 0
       0      .1       0   170.9    .045       0   200.2     .08       0
Bank Sta=170.9,200.2
XS Rating Curve= 0 ,0
Exp/Cntr=0.3,0.1

Type RM Length L Ch R = 1 ,9368.3  ,209.5,209.1,208.6
XS GIS Cut Line= 4
      1672755.14      745137.505     1672725.626      745180.908
     1672581.528      745436.117     1672564.167      745611.464
#Sta/Elev= 30
       0 1023.12    17.5 1019.56      35 1015.78    43.7 1013.09    52.5 1008.49
    62.3 1001.12      72  993.16    81.8  985.56    91.6  982.32    92.7  982.26
   101.3  981.81   107.7   981.8   111.1   981.8   130.6   981.8   140.4  981.92
     160  983.28   169.7  983.82     199  985.11   218.6  985.76   247.9  985.94
   267.4  986.26   277.2  986.67     287  987.21   306.5  988.55     326  990.07
   355.4  992.68   384.7  995.62   492.4 1007.27     512 1009.54   521.8  1010.8
#Mann= 3 , 0 , 0
       0      .1       0    92.7    .045       0   111.1     .08       0
Bank Sta=92.7,111.1
XS Rating Curve= 0 ,0
Exp/Cntr=0.3,0.1

Type RM Length L Ch R = 1 ,9159.2  ,225.3,225.9,226.3
XS GIS Cut Line= 4
     1672590.209      745087.158     1672546.806      745128.825
      1672388.82      745417.019     1672362.778      745620.144
#Sta/Elev= 30
       0 1024.44    25.8 1021.89      43 1019.76    51.6 1018.31    60.2 1015.52
    69.8 1008.62    79.5  997.37    89.2  986.99    98.8  982.57   108.5   981.8
   118.2  981.81   137.5  981.95   195.5  983.51   224.5  984.56   253.5  985.81
   311.5   988.9   369.5   991.5   388.8     992   418.1  992.24   427.8  992.46
   457.1  993.68   486.3   995.1   505.8   996.4   525.4  998.02   535.1  998.96
   554.6 1001.22   564.4 1002.63   574.1 1004.32   583.9 1006.14   593.6 1008.14
#Mann= 3 , 0 , 0
       0      .1       0   118.2    .045       0   137.5     .07       0
Bank Sta=118.2,137.5
XS Rating Curve= 0 ,0
Exp/Cntr=0.3,0.1

Type RM Length L Ch R = 1 ,8933.4  ,271.6,272.8,273.8
XS GIS Cut Line= 4
     1672361.042      744981.255     1672340.209      745078.478
     1672230.834      745271.186      1672130.14      745432.644
#Sta/Elev= 28
       0 1032.61    18.1 1028.04    36.2 1023.11    54.2  1017.9    63.3  1014.9
    72.3 1011.15    81.4 1006.52    90.4 1001.44    99.4  996.07   109.1  990.62
   118.7  986.17   128.3   983.4     138  982.14   147.6   981.8     152   981.8
   176.5   981.8   205.4  981.84     215  982.04   224.7  982.69   272.8  987.52
   282.5  988.45   301.7  990.09   330.5  992.33   406.6  997.89   425.7     999
   444.7  999.96   482.8 1001.56   511.3 1002.63
#Mann= 3 , 0 , 0
       0      .1       0     152    .045       0   176.5      .1       0
Bank Sta=152,176.5
XS Rating Curve= 0 ,0
Exp/Cntr=0.3,0.1

Type RM Length L Ch R = 1 ,8660.6  ,159.9,165.6,171.1
XS GIS Cut Line= 4
     1672180.487      744936.117     1672131.876      744976.047
     1671984.306       745206.95     1671965.209      745397.922
#Sta/Elev= 26
       0 1006.79      27 1003.83      36  1002.7    44.9 1001.15    53.9   998.9
    62.9  996.03    72.7  992.72    92.3  984.92   102.1  982.77   111.8  982.18
   121.6  981.97   141.2   981.8   199.9   981.8   219.5   981.8   229.3   981.9
   239.1  982.41   248.9  983.11   258.6  983.97   268.4  984.91   307.6  989.23
   317.4   990.2   336.9  991.74   365.7   993.7   404.1  996.16   490.5 1001.52
   528.9  1003.8
#Mann= 3 , 0 , 0
       0      .1       0   199.9    .045       0   229.3      .1       0
Bank Sta=199.9,229.3
XS Rating Curve= 0 ,0
Exp/Cntr=0.3,0.1

Type RM Length L Ch R = 1 ,8495.1  ,67.8,67.8,67.9
XS GIS Cut Line= 6
      1672201.32      744783.339     1672078.056      744880.561
     1672048.542      744899.658     1671937.431      745012.505
     1671885.348      745094.103     1671835.001      745345.839
#Sta/Elev= 30
       0 1008.77     9.8 1006.85    19.6  1005.1    39.2 1001.92    58.9  999.01
    78.5   996.5    98.1  994.61   117.7  992.99   147.2     991   174.6  989.43
   183.4  988.67   192.1  987.75   210.8  985.36   220.1  983.89   229.4  982.89
   238.7   982.4     248   982.1   266.7  981.82   276.6  981.99   303.9  983.66
   313.2   983.9   360.2  983.35   369.9  983.33   379.6  983.49   532.9  989.26
   542.4  989.79   580.4  992.41     609  994.23   656.5  997.04     704 1000.68
#Mann= 3 , 0 , 0
       0      .1       0     248    .045       0   276.6     .08       0
Bank Sta=248,276.6
XS Rating Curve= 0 ,0
Exp/Cntr=0.3,0.1

Type RM Length L Ch R = 1 ,8427.2  ,53.5,50.7,47.9
XS GIS Cut Line= 6
     1672159.653      744731.255      1672036.39      744828.478
     1672006.876      744847.575     1671895.765      744960.422
     1671843.681      745042.019     1671793.334      745293.755
#Sta/Elev= 30
       0  995.72    29.4   993.6    68.7  991.48    78.5  990.63    98.1  988.55
   107.9  987.78   137.4  986.45   165.8  985.53   220.1  982.21   238.7  980.91
   256.6  980.58   257.4  980.57   271.6  980.75   341.2  981.11   369.9  981.62
   389.2  982.22   408.6  983.06   437.6  984.73   456.8  985.57   561.4  987.57
   570.9  987.94   580.4  988.65   599.4  990.69     609  991.49   618.5  991.96
   637.5  992.44     647  992.89   675.5  994.94   694.5  996.61     704  997.63
#Mann= 3 , 0 , 0
       0      .1       0   256.6    .045       0   271.6     .06       0
Bank Sta=256.6,271.6
XS Rating Curve= 0 ,0
Exp/Cntr=0.3,0.1

Type RM Length L Ch R = 1 ,8376.5  ,258,261.9,267.1
XS GIS Cut Line= 4
     1671996.459      744668.755     1671965.209      744804.172
     1671710.001      745137.505     1671578.056      745203.478
#Sta/Elev= 30
       0 1000.39    27.8   998.8    55.6  998.26    74.1  997.59   129.7  994.05
     139     993   148.7  991.21     178  984.74   187.8  982.77   197.6  980.91
   207.9   979.6   217.1  979.17   236.6  979.41   334.2  981.53     383  983.32
   422.1  984.18   470.9  985.53   500.2  986.48   539.3  988.29     549  989.17
   558.8  991.22   578.5  996.66   588.3   998.9     608 1002.87   617.8  1004.6
   627.6 1006.02   637.5 1007.26   647.3 1007.98     667 1008.91   706.3 1011.24
#Mann= 3 , 0 , 0
       0      .1       0   207.9    .045       0   236.6     .06       0
Bank Sta=207.9,236.6
XS Rating Curve= 0 ,0
Exp/Cntr=0.3,0.1

Type RM Length L Ch R = 1 ,8114.6  ,180.6,175.7,169.1
XS GIS Cut Line= 4
     1671867.987      744576.742     1671803.751      744634.033
     1671612.778      744781.603     1671503.403      744929.172
#Sta/Elev= 30
       0  1007.8    38.2 1001.11    47.8  999.67      67  997.85    76.5  996.06
    86.1  993.14     115  983.67   124.7  980.83   134.3   978.9   153.6   978.8
   163.3  978.83     173  978.99   201.9  980.74   221.2  981.61   240.5  982.24
   269.5  982.69   279.2  982.99   288.8  983.82   298.5  985.52   308.1  988.15
   327.4  993.85   337.1  996.33   346.8  998.38   356.4 1000.06   424.1 1009.18
   453.1 1012.86   472.4 1015.14   482.1 1016.19   501.4 1018.11   511.1 1018.89
#Mann= 3 , 0 , 0
       0      .1       0   134.3    .045       0   163.3      .1       0
Bank Sta=134.3,163.3
XS Rating Curve= 0 ,0
Exp/Cntr=0.3,0.1

Type RM Length L Ch R = 1 ,7938.9  ,264.2,267.2,269.4
XS GIS Cut Line= 4
     1671706.528      744453.478      1671670.07      744505.561
     1671527.709      744691.325      1671473.89      744816.325
#Sta/Elev= 26
       0 1014.27     9.1 1012.31    18.2 1009.83    36.3 1004.27    54.5  998.78
    83.1  989.97   102.6  984.36   112.3  981.69   122.1  979.58   127.8  979.12
   131.8   978.8   151.3   978.8   170.8  978.82   180.6  978.92   190.4   979.4
   200.1  980.41   229.4  984.11   239.1  985.41   248.9  986.92   268.4  990.53
   278.1   992.1   307.3  996.62   336.5 1001.02   365.7 1005.09   404.6 1009.93
   433.7 1013.88
#Mann= 3 , 0 , 0
       0      .1       0   127.8    .045       0   151.3      .1       0
Bank Sta=127.8,151.3
XS Rating Curve= 0 ,0
Exp/Cntr=0.3,0.1

Type RM Length L Ch R = 1 ,7671.7  ,164.5,159.7,154.9
XS GIS Cut Line= 4
     1671552.015      744293.755     1671484.306      744335.422
     1671308.959      744517.714     1671215.209      744670.492
#Sta/Elev= 27
       0 1008.26    17.7 1006.46      53 1003.07    61.8 1002.08    70.7 1000.69
    79.5  997.33    89.2  992.17      99  985.79   108.7  979.97   118.4   976.4
   128.1  975.57   137.9  976.09     206  980.29   225.4  981.61   244.9  983.12
   274.1  985.63   283.8  986.49   303.2  988.45   322.7  990.73     389  998.82
   407.9 1000.97   417.4 1002.82   426.8 1006.15   436.2 1009.33   445.6 1010.65
   483.4 1013.67   511.7 1015.82
#Mann= 3 , 0 , 0
       0      .1       0   118.4    .045       0   137.9      .1       0
Bank Sta=118.4,137.9
XS Rating Curve= 0 ,0
Exp/Cntr=0.3,0.1

Type RM Length L Ch R = 1 ,7512.1  ,311.7,279.8,248.3
XS GIS Cut Line= 4
     1671585.102      744067.555     1671352.362      744226.047
     1671220.417      744439.589     1671190.903      744531.603
#Sta/Elev= 30
       0  1041.3    29.1 1035.54      68 1026.92   106.8 1019.77   116.5 1018.53
   135.9 1017.54   145.6 1016.57   184.5 1011.96     233 1005.57   252.4 1002.59
   271.9  999.06   281.6  996.96   300.9  992.03   310.5  988.79   320.2  984.77
   329.8  980.33   339.5  976.79   349.2  975.48   358.8   975.4   366.8  975.45
   378.1  975.81   387.8  976.56   445.7  981.78   474.7  984.61   513.3   988.9
   580.9  997.77   590.6  999.47   609.9 1003.82   619.6 1005.37   629.2 1006.28
#Mann= 3 , 0 , 0
       0      .1       0   339.5    .045       0   366.8      .1       0
Bank Sta=339.5,366.8
XS Rating Curve= 0 ,0
Exp/Cntr=0.3,0.1

Type RM Length L Ch R = 1 ,7232.3  ,144.7,139.1,132.2
XS GIS Cut Line= 5
     1670853.765      743922.155      1670943.06      744119.265
     1670970.417      744142.714     1671185.695      744338.894
     1671190.903      744430.908
#Sta/Elev= 30
       0 1097.83    19.7 1089.96    39.3 1081.18    49.2 1077.36      59 1074.46
    78.7 1069.07   127.9 1056.23   137.7 1053.41   147.5 1050.07   157.4 1045.93
   206.6  1020.2   216.4 1015.02   234.4 1004.22   243.4   999.4   252.4  994.98
   262.1  990.65   271.8   987.2   291.3  981.39     301  979.44   310.7  978.61
   339.8  976.89   369.8  974.79   388.3  973.87     398  973.76   446.6  974.86
   456.3  975.27   475.7  976.46   543.7  981.44   580.6  985.03   635.8  991.66
#Mann= 3 , 0 , 0
       0      .1       0   369.8    .045       0     398      .1       0
Bank Sta=369.8,398
XS Rating Curve= 0 ,0
Exp/Cntr=0.3,0.1

Type RM Length L Ch R = 1 ,7093.2  ,57.3,57.3,57.3
XS GIS Cut Line= 3
     1670831.528      744231.255     1670890.556      744259.033
      1671161.39      744413.547
#Sta/Elev= 30
       0 1012.01     9.3 1011.08    18.6 1009.68    46.6 1004.32    55.9 1002.88
      75 1000.32    94.5  998.17     114  996.15   123.7  995.23   143.2  993.59
   152.9  992.01   172.4  987.01   182.2  985.07   191.9  984.01   201.6  983.37
   211.4  982.82   221.1  982.72   230.9  981.52   240.6  978.74   247.2  976.17
   250.4  974.92   260.1  973.99   269.9  977.85   279.6  983.66   289.4  987.81
   299.1  989.06   308.8  989.48   318.6  989.58   347.8  990.34     377  990.88
#Mann= 3 , 0 , 0
       0      .1       0   247.2    .045       0   269.9      .1       0
Bank Sta=247.2,269.9
XS Rating Curve= 0 ,0
Exp/Cntr=0.3,0.1

Type RM Length L Ch R = 1 ,7035.9  ,176.2,192.3,208.6
XS GIS Cut Line= 3
     1670808.959      744283.339     1670867.987      744311.117
      1671138.82       744465.63
#Sta/Elev= 30
       0 1005.78    18.6  1005.8    37.3 1005.09    46.6 1004.32      75 1001.05
    84.7 1000.11    94.5  999.26   123.7  997.18   133.4  994.65   143.2  991.14
   152.9  986.98   162.7  983.85   172.4  982.53   201.6  979.42   211.4  978.16
   221.1  976.58   240.6  973.09   250.4  971.66   260.1  971.81     266  973.82
   269.9  975.15   279.6  979.06   299.1  986.58   308.8  990.11   318.6  993.36
   328.3  996.24   338.1  998.57   347.8 1000.36   367.3  1002.9     377 1003.66
#Mann= 3 , 0 , 0
       0      .1       0   240.6    .045       0     266      .1       0
Bank Sta=240.6,266
XS Rating Curve= 0 ,0
Exp/Cntr=0.3,0.1

Type RM Length L Ch R = 1 ,6843.6  ,216.7,236.9,257.1
XS GIS Cut Line= 4
     1670831.528      744328.478     1670847.153      744385.769
     1670918.334      744602.783     1670927.015      744720.839
#Sta/Elev= 29
       0  1005.3     8.5  1004.3    33.9  1000.9    42.4  999.86    50.9  998.47
    59.4  996.16    68.9  992.59    87.9  983.85    97.4  980.67     107  979.12
   116.5   978.1     126  976.86     145  973.83   164.1  970.49   173.6   969.1
   183.1  968.29   192.6  968.03   202.1  968.09   211.6  968.89   221.2  971.22
   240.2  976.72   259.2  981.98   268.7  984.94   296.9  993.19     306  996.05
   315.1  998.78   324.2 1000.95   333.3 1002.23   406.2 1007.41
#Mann= 3 , 0 , 0
       0      .1       0   183.1    .045       0   211.6      .1       0
Bank Sta=183.1,211.6
XS Rating Curve= 0 ,0
Exp/Cntr=0.3,0.1

Type RM Length L Ch R = 1 ,6606.7  ,278.5,266.7,254.8
XS GIS Cut Line= 3
     1670762.084      744302.436      1670723.89      744345.839
     1670574.584      744588.894
#Sta/Elev= 26
       0 1003.23    38.5  999.41    48.2  998.12    57.8  995.19    67.6  989.92
    77.5  983.23    87.3  976.25    97.2  970.74     107  968.46   116.8     968
   143.6     968     166     968   175.8  968.76   185.7   973.2   195.5  980.61
   205.4  988.24   215.2  994.55     225  998.39   234.9  999.87   254.5  1001.4
     284  1003.5   303.7 1004.75   313.6 1005.25   323.4 1005.69   333.2 1006.03
   343.1 1006.25
#Mann= 3 , 0 , 0
       0      .1       0   143.6    .045       0     166      .1       0
Bank Sta=143.6,166
XS Rating Curve= 0 ,0
Exp/Cntr=0.3,0.1

Type RM Length L Ch R = 1 ,6340    ,272.5,252,231.2
XS GIS Cut Line= 4
     1670470.417      744118.408     1670466.945        744175.7
     1670460.001      744441.325     1670465.209       744496.88
#Sta/Elev= 23
       0 1016.78     9.6  1013.9    19.1 1010.85    28.7 1007.32    47.8  999.56
    77.1  988.08    96.8  980.23   116.4  972.28   126.3  969.06   136.1     968
   155.1     968   175.5     968   214.9  968.02   224.7  968.35   234.5     970
   244.4  973.44   273.9  983.99   303.4  994.42   313.3  997.71   323.1 1000.36
   332.4 1001.45   360.3 1001.39   378.9 1001.44
#Mann= 3 , 0 , 0
       0      .1       0   155.1    .045       0   175.5      .1       0
Bank Sta=155.1,175.5
XS Rating Curve= 0 ,0
Exp/Cntr=0.3,0.1

Type RM Length L Ch R = 1 ,6087.9  ,148.6,148.7,148.6
XS GIS Cut Line= 4
     1670046.806      744189.589     1670149.237      744297.228
     1670343.681      744455.214     1670444.376      744502.089
#Sta/Elev= 30
       0 1034.01    18.6 1032.01    37.2 1028.49    74.3 1016.03    92.9 1009.19
   120.7  998.05   139.3  991.98   148.6  990.05   167.9  987.52   187.1   986.3
     216  985.47   225.7  983.73   235.3  980.27     245  975.81   254.6  970.23
   260.5  968.95   264.2  968.15   273.9     968   283.5     968   293.1     968
   302.8  968.97   312.4  972.02   331.7  980.94   341.3  984.44   370.2  991.21
   389.5  995.06   408.4  997.45   445.4 1000.45   491.7 1000.06   510.2 1000.42
#Mann= 3 , 0 , 0
       0      .1       0   260.5    .045       0   283.5      .1       0
Bank Sta=260.5,283.5
XS Rating Curve= 0 ,0
Exp/Cntr=0.3,0.1

Type RM Length L Ch R = 1 ,5939.2  ,145.9,148.4,150.8
XS GIS Cut Line= 4
     1669932.223      744286.811     1670034.653       744394.45
     1670229.098      744552.436     1670329.792      744599.311
#Sta/Elev= 30
       0 1015.23    18.6 1015.24    37.2  1012.5    46.4 1010.47    83.6 1000.92
   120.7  991.88     130  988.83   139.3   983.5   148.6   976.9   158.2  971.04
   167.9  967.36   177.5  965.14   187.1  964.22   254.6  962.77   264.2   961.5
   273.9  958.53   283.5  960.12   287.2  962.36   302.8  971.63     322  980.82
   331.7  983.97   341.3  986.37   350.9   988.1   360.6  989.09   399.1  991.89
   426.9  996.84   436.2  998.07   445.4  998.78   454.7  999.13   510.2   998.6
#Mann= 3 , 0 , 0
       0      .1       0   254.6    .045       0   287.2      .1       0
Bank Sta=254.6,287.2
XS Rating Curve= 0 ,0
Exp/Cntr=0.3,0.1

Type RM Length L Ch R = 1 ,5790.8  ,279.7,280.9,282
XS GIS Cut Line= 3
     1669896.633       744394.45     1669934.827      744482.992
     1670113.646      744663.547
#Sta/Elev= 29
       0  998.49     9.6  996.28    19.3  993.88    28.9  990.96    38.6  987.22
    48.2  982.97    57.9  978.51    67.5   973.7    77.1   969.1    86.8     966
    96.4  964.54   106.2  963.89   145.3  961.68   184.4  959.86   194.2  958.94
   203.9  957.05   210.7  955.57   213.7  954.92   223.5  954.85   225.7  955.59
   233.3  958.13     243  963.48   262.6   974.9   272.4  980.44   282.1  985.65
   291.9  989.84   301.7  992.02   311.4  993.04   350.6  995.93
#Mann= 3 , 0 , 0
       0      .1       0   210.7    .045       0   225.7      .1       0
Bank Sta=210.7,225.7
XS Rating Curve= 0 ,0
Exp/Cntr=0.3,0.1

Type RM Length L Ch R = 1 ,5509.9  ,345.2,345.6,344.5
XS GIS Cut Line= 2
     1669640.006      744563.865     1669906.934      744862.043
#Sta/Elev= 24
       0  965.71     9.8  961.38    19.5  958.63    29.3  957.73    58.6  956.79
    78.1  956.38   126.9  955.86   165.9  955.61   195.2  955.33     205  955.13
   214.7     954   224.5   951.8   234.3  950.29   243.4  952.11     244  952.23
   253.8  956.79   292.8  977.87   312.4  988.27   322.1  992.53   331.9  994.65
   341.6  995.95   351.4  997.02   370.9  998.72   400.2  1001.1
#Mann= 3 , 0 , 0
       0      .1       0   224.5    .045       0   243.4      .1       0
Bank Sta=224.5,243.4
XS Rating Curve= 0 ,0
Exp/Cntr=0.3,0.1

Type RM Length L Ch R = 1 ,5164.3  ,188.8,189.6,191.1
XS GIS Cut Line= 2
     1669395.215      744662.824     1669668.652      745001.365
#Sta/Elev= 29
       0  995.73    19.3  980.36    38.7  965.03    48.4  958.09      58  952.97
    67.7  950.03    77.4   947.6      87  945.84    96.7  945.22   106.3   945.2
   121.3   945.2   145.1  945.28   154.7  945.47   164.4  945.93   203.1  948.13
   212.8  948.81   232.1  950.35   251.4  952.28   319.1  959.76   328.8  961.11
   338.5   964.2   348.1  969.82   357.8  977.56   367.5  984.18   377.2   987.8
   386.8  989.37   406.2  991.16   415.8  991.83   435.2  992.98
#Mann= 3 , 0 , 0
       0      .1       0    96.7    .045       0   121.3      .1       0
Bank Sta=96.7,121.3
XS Rating Curve= 0 ,0
Exp/Cntr=0.3,0.1

Type RM Length L Ch R = 1 ,4974.8  ,405.7,407.9,409.4
XS GIS Cut Line= 2
     1669241.569      744765.688     1669503.288      745074.282
#Sta/Elev= 24
       0 1013.95    48.2   979.9    77.1  959.12    86.7  952.34    96.3  946.74
     106  943.93   109.9  943.55   115.6     943   124.9  942.91   134.9  943.14
   144.5  943.61   154.2  944.22     212  947.49   240.8   949.5   250.5   949.9
   260.1  949.99   269.8  950.28     289  951.78   317.9  953.91   327.6  954.77
   337.2  955.79   356.5  958.06   385.4  961.61   404.6  964.34
#Mann= 3 , 0 , 0
       0      .1       0   109.9    .045       0   134.9      .1       0
Bank Sta=109.9,134.9
XS Rating Curve= 0 ,0
Exp/Cntr=0.3,0.1

Type RM Length L Ch R = 1 ,4566.9  ,261.1,269.5,278.2
XS GIS Cut Line= 4
     1668968.131       745048.24     1668999.381      745100.324
     1669126.986      745280.011     1669257.194       745454.49
#Sta/Elev= 30
       0  975.21    60.7  948.14    79.9  939.76    89.5  936.52    99.1  935.21
   108.6   935.1   118.2  935.14   127.8  935.47   137.4  936.67   166.1  941.47
   185.3  943.53   204.5  945.04   223.6  946.17   242.8  946.97   290.6  948.34
   309.5  949.12     319  949.94   337.9  952.71   356.8   955.2   366.3  956.16
   394.7  958.29   413.6  959.97   423.1  961.22   432.6  962.86     442  964.88
   451.5  967.48     461     971   470.4  974.94   479.9  977.48   498.8  979.12
#Mann= 3 , 0 , 0
       0      .1       0    99.1    .045       0   118.2      .1       0
Bank Sta=99.1,118.2
XS Rating Curve= 0 ,0
Exp/Cntr=0.3,0.1

Type RM Length L Ch R = 1 ,4297.3  ,286.1,294.3,299.9
XS GIS Cut Line= 4
     1668770.215      745112.043     1668771.517      745190.168
     1668824.902      745411.522     1668841.829      745656.313
#Sta/Elev= 30
       0  974.33     9.8  970.95    48.8  956.78    87.6  942.98   106.6  936.47
   116.1  934.21   125.6  934.41   135.1  935.73   144.6  937.76     154  939.29
   163.5  940.35     192  942.61   220.4  943.92   248.9  944.45   305.8  944.24
   354.9  944.98   384.4  945.11   394.2   945.3     404  945.75   423.6  947.31
   443.2  949.43   462.9     952   472.7  953.94   492.3  958.85   502.1  960.21
     512  961.16   521.8  963.11   531.6   966.2   541.4  969.85   551.2  973.77
#Mann= 3 , 0 , 0
       0      .1       0   106.6    .045       0   135.1      .1       0
Bank Sta=106.6,135.1
XS Rating Curve= 0 ,0
Exp/Cntr=0.3,0.1

Type RM Length L Ch R = 1 ,4003.1  ,108.1,104.4,103
XS GIS Cut Line= 2
     1668516.309       745110.74     1668525.423      745619.855
#Sta/Elev= 30
       0  964.59    19.6  961.71    29.4  959.86    39.2  955.86    58.8   941.5
    68.6  937.88    78.3  937.15    97.9  936.87   117.5  936.73   166.5  935.98
   176.3  935.71   195.8     935   205.6  934.46   215.4  933.77   225.2  933.52
     235   933.5   244.8  933.66   254.6  935.34   264.4   937.5   274.2  938.59
   313.4  940.41   332.9  941.04   362.3   941.5   430.9  941.87   450.4  942.05
   460.2  943.65     470  947.44   479.8  952.09   499.4  961.88   509.2  965.09
#Mann= 3 , 0 , 0
       0      .1       0   225.2    .045       0   244.8      .1       0
Bank Sta=225.2,244.8
XS Rating Curve= 0 ,0
Exp/Cntr=0.3,0.1

Type RM Length L Ch R = 1 ,3898.7  ,31.8,31.6,31.8
XS GIS Cut Line= 2
     1668405.631      745109.438     1668435.579      745618.553
#Sta/Elev= 30
       0  956.92    29.4  951.66    39.2  949.64      49  945.91    58.8  940.21
    68.6  935.93    78.5  934.82   127.5  935.76   176.5  936.02   186.3   936.2
   196.2  936.26     206  935.72   215.8  934.77   225.6  933.97   235.4  933.59
   245.2  933.52     255  934.21   264.8  935.93   274.6   937.2   284.4  937.43
   294.2  937.51   353.1  938.63   431.5  939.65   441.3  939.92   451.2  940.32
     461  941.24   470.8  943.56   480.6  947.32   500.2  956.07     510  960.31
#Mann= 3 , 0 , 0
       0     .08       0   225.6    .045       0     255      .1       0
Bank Sta=225.6,255
XS Rating Curve= 0 ,0
Exp/Cntr=0.3,0.1

Type RM Length L Ch R = 1 ,3867.1  ,65.1,66.3,66.2
XS GIS Cut Line= 2
     1668374.381      745112.043     1668404.329      745621.157
#Sta/Elev= 30
       0  955.65    19.6  952.04    29.4  949.31    39.2     945      49   939.8
    58.8  935.86    68.6  934.28    78.5  934.12   127.5  934.97   196.2  935.54
     206   935.2   215.8   934.3   225.6  933.18   235.4  932.29   245.2   932.7
     255  934.93   264.8  937.16   274.6  937.99   284.4  937.87     304  936.99
   313.8  936.86   323.6  936.95   362.9  938.37   372.7  938.58   421.7  938.84
   451.2  940.04     461  940.83   470.8  942.87   480.6  946.53     510   959.5
#Mann= 3 , 0 , 0
       0     .08       0   215.8    .045       0     255      .1       0
Bank Sta=215.8,255
XS Rating Curve= 0 ,0
Exp/Cntr=0.3,0.1

Type RM Length L Ch R = 1 ,3800.7  ,160.8,166.6,172.8
XS GIS Cut Line= 3
     1668326.204      745083.397     1668320.996      745117.251
     1668331.413       745635.48
#Sta/Elev= 30
       0  959.06     8.6   957.3    17.1  955.14    25.7  952.18    53.8  939.63
    63.6  935.93    73.4  933.59    83.2  932.63    92.9  932.46   171.2   932.3
   200.5  931.78   220.1  931.06   239.6  930.06   249.4  930.11   256.6  931.15
   259.2  931.53   278.8  936.41   288.5   937.8   298.3  938.36   308.1  938.31
   347.2  936.23     357   936.3   396.1  938.41   464.6   938.5   484.1  939.11
   493.9  939.89   503.7  942.04   513.5  945.63   542.8  957.82   552.6  960.56
#Mann= 3 , 0 , 0
       0     .08       0   220.1    .045       0   256.6      .1       0
Bank Sta=220.1,256.6
XS Rating Curve= 0 ,0
Exp/Cntr=0.3,0.1

Type RM Length L Ch R = 1 ,3634.1  ,208.8,217.2,225.5
XS GIS Cut Line= 4
     1668224.642      745062.563      1668192.09      745171.938
     1668115.267      745500.063     1668093.131      745716.209
#Sta/Elev= 30
       0  950.34     9.5  946.97    28.5  939.26      38   936.3    47.6   934.9
    57.1  934.54    85.6  934.29   104.6  933.82   152.6  931.27   181.5   930.6
   191.1  930.04   210.4  928.31     220  927.42   229.7  927.08   239.3   927.5
   277.8  930.88   297.1  931.98   316.3  932.62   393.3  933.49   460.6  936.53
   498.4  937.83   507.8  938.88   517.2  941.56   536.1  948.91   545.6  951.25
     555  952.26   564.5   953.9   573.9  957.19   630.6  981.32   668.4  997.89
#Mann= 3 , 0 , 0
       0      .1       0   210.4    .045       0   239.3      .1       0
Bank Sta=210.4,239.3
XS Rating Curve= 0 ,0
Exp/Cntr=0.3,0.1

Type RM Length L Ch R = 1 ,3417    ,271.1,269.1,266.8
XS GIS Cut Line= 4
     1668093.131       745041.73     1668048.861      745074.282
     1667852.246      745362.043     1667801.465      745484.438
#Sta/Elev= 30
       0  949.88     9.2  943.83    18.3  937.29    27.5  932.86    36.6  931.86
    64.6  931.94    74.3   931.8    93.7  931.04   122.7  929.24   171.1  925.44
   180.8  924.83   190.5  924.71   200.2   925.3   229.2  927.76   248.6  928.97
   267.9  929.81   306.7  930.71   345.4  931.93   403.5  932.14   412.9  932.53
   422.4  933.23   431.9  934.47   441.3  936.48   460.3  942.17   469.7  944.49
   479.2  945.56   498.1  946.26   507.6  947.23     517  949.28     536  954.92
#Mann= 3 , 0 , 0
       0      .1       0   171.1    .045       0   200.2      .1       0
Bank Sta=171.1,200.2
XS Rating Curve= 0 ,0
Exp/Cntr=0.3,0.1

Type RM Length L Ch R = 1 ,3147.9  ,270.2,269.2,268.2
XS GIS Cut Line= 3
     1667801.852      744863.742     1667781.934      744984.438
     1667593.131      745311.261
#Sta/Elev= 30
       0  968.48    94.1  950.98   103.5  949.07   112.9  946.38   122.3  942.09
   141.7  929.88   151.4  925.04     161  922.55   170.7  921.65   180.4  921.42
   188.5  921.41   199.8  921.61   203.5  921.98   209.4  922.56   219.1   924.5
   228.8  926.67   238.5  928.98   267.5  936.65   277.2  939.08   286.8  940.62
   296.5  941.14   325.6  941.76   344.9  941.98   393.3  942.25   412.7  942.08
   441.7  941.14   451.4  940.91     461   940.8   490.1  940.83   499.8  940.76
#Mann= 3 , 0 , 0
       0      .1       0   180.4    .045       0   203.5      .1       0
Bank Sta=180.4,203.5
XS Rating Curve= 0 ,0
Exp/Cntr=0.3,0.1

Type RM Length L Ch R = 1 ,2878.6  ,437.2,427.1,417
XS GIS Cut Line= 3
     1667593.518      744792.128     1667544.954      744872.459
      1667354.85      745244.855
#Sta/Elev= 30
       0  967.89    37.6   960.4    56.3  955.86    65.7  953.21    75.1   950.4
    84.5  946.69    93.9  940.36   103.6  930.57   113.3  923.09     123  920.45
   132.8  920.06   142.5  920.09   149.2  920.34   152.2  920.45   181.4   922.4
   191.1  923.54   200.8  925.38   210.6  927.54   220.3  929.78     230  931.76
   239.7  932.73   249.4  932.61   259.2  932.62   307.8  933.39   317.5  933.48
   366.1  933.51   434.2  933.77   473.1  933.83   502.3   933.7     512  933.96
#Mann= 3 , 0 , 0
       0      .1       0     123    .045       0   149.2      .1       0
Bank Sta=123,149.2
XS Rating Curve= 0 ,0
Exp/Cntr=0.3,0.1

Type RM Length L Ch R = 1 ,2451.6  ,231.2,206.5,186.1
XS GIS Cut Line= 4
     1667154.583      744564.516     1667121.777       744697.98
     1667115.267      744912.824     1667274.121       745104.23
#Sta/Elev= 30
       0  953.49     9.8  951.72    29.4   948.7    68.7  943.75    78.5  942.05
    88.4   939.9   117.8   932.6   137.4  927.99   147.2  925.91     157  924.12
   176.5  921.43   205.8  918.11   215.6  917.48   225.4  917.75   232.3  918.91
   235.1  919.38   244.9  921.81   254.7  923.69   264.4  924.79   274.2  925.43
     284   925.6   313.3  924.48   323.1  924.46     362  925.87   381.1  926.15
   409.8  926.04   457.6  926.29   495.9  925.57   562.8  928.35   601.1  929.33
#Mann= 3 , 0 , 0
       0      .1       0   205.8    .045       0   232.3      .1       0
#XS Ineff= 2 , 0
                          282.11          930.92
Permanent Ineff=
       F       F
Bank Sta=205.8,232.3
XS Rating Curve= 0 ,0
Exp/Cntr=0.3,0.1

Type RM Length L Ch R = 1 ,2245.1  ,89.5,88.5,83.7
XS GIS Cut Line= 6
     1666663.444      744789.126     1666839.225      744808.657
     1666891.309      744828.188     1666955.111      744864.647
     1667033.236      744929.751     1667186.881      745114.647
#Sta/Elev= 30
       0  977.53    19.6  969.38    39.3  961.68    49.1  957.97    68.8  950.99
    78.6  947.74    98.3  941.69   108.1  938.95   117.9  936.68   127.7  935.05
     167  930.87   176.9   929.4   195.4  925.49   204.7  923.97     214  922.88
   241.7  920.68   269.2  919.53   278.4  918.75   287.6  917.64   296.8  916.82
   313.2   916.6   324.5  917.46     343  920.53   407.7  922.58   427.1  922.71
   504.7  922.39   562.6   922.9   591.1  923.49   610.1  924.22   648.1  926.61
#Mann= 3 , 0 , 0
       0     .06       0   287.6    .045       0   324.5     .08       0
Bank Sta=287.6,324.5
XS Rating Curve= 0 ,0
Exp/Cntr=0.3,0.1

Type RM Length L Ch R = 1 ,2156.6  ,153.5,154.1,154
XS GIS Cut Line= 6
     1666645.215      744875.063     1666820.996      744894.595
     1666873.079      744914.126     1666936.881      744950.584
     1667015.006      745015.688     1667168.652      745200.584
#Sta/Elev= 30
       0  956.34    19.6  946.91    49.1  933.24      59  928.99    68.8   925.6
    78.6   923.6    98.3  921.77   117.9  918.91   127.7   917.8   137.6  916.96
   147.4  916.52     167   916.4     306   916.4   315.2  916.67     319 917.148
   333.7   918.8   352.2  919.34   370.7   919.6   379.9  920.19   389.2  922.56
   398.4  925.94   407.7  929.99   417.4  933.66   436.8  938.57   446.5  940.03
   514.4  945.17   543.5  947.06   600.6  951.69   629.1  954.96   648.1  957.84
#Mann= 3 , 0 , 0
       0      .1       0     167    .045       0     319      .1       0
Bank Sta=167,319
XS Rating Curve= 0 ,0
Exp/Cntr=0.3,0.1

Type RM Length L Ch R = 1 ,2002.5  ,228.5,217.7,206.8
XS GIS Cut Line= 4
     1666517.828      744934.525     1666642.611      744959.699
     1666891.309      745092.511     1666987.663      745152.407
#Sta/Elev= 30
       0 1014.01     9.8 1008.27    29.4  997.12    39.2  991.28      49  984.69
    58.8  977.49    88.1  954.74    97.9  947.21   107.7  939.88   117.5  932.94
   127.3  927.14     137  923.71   146.7  922.12   156.5  920.08   166.2  917.37
   175.9  916.48   185.6   916.4   360.6   916.4   370.4   916.5     373916.7413
   380.1   917.4   389.8  920.33   418.7  932.49     447  943.91   475.4  954.56
   484.9  957.74   494.3  960.72   503.8   963.3   513.2  964.95   522.7  966.04
#Mann= 3 , 0 , 0
       0      .1       0   175.9    .045       0     373      .1       0
Bank Sta=175.9,373
XS Rating Curve= 0 ,0
Exp/Cntr=0.3,0.1

Type RM Length L Ch R = 1 ,1784.8  ,301.2,313.4,325.4
XS GIS Cut Line= 3
     1666572.298      745261.782     1666630.892      745257.876
      1666979.85      745261.782
#Sta/Elev= 19
       0  954.45    19.6  940.26    29.4  933.43    39.2  928.12    48.9  925.82
    58.7   924.4    68.4  921.32      73919.7171    78.1  917.94    87.8   916.4
     260   916.4     272   916.4   281.7  916.88   291.4  920.23   330.2  935.98
   349.5  943.91   359.2  947.98   388.3  959.93   407.7  968.05
#Mann= 3 , 0 , 0
       0      .1       0      73    .045       0     260      .1       0
Bank Sta=73,260
XS Rating Curve= 0 ,0
Exp/Cntr=0.3,0.1

Type RM Length L Ch R = 1 ,1471.4  ,399.1,407.6,415.9
XS GIS Cut Line= 4
     1666568.392      745493.553     1666632.194      745522.199
     1666804.069      745625.063     1666913.444      745648.501
#Sta/Elev= 25
       0   943.4     8.7  942.32    17.5   940.3    26.2  937.58    43.7  931.72
    52.4  928.89    69.9  923.39    79.5  920.53      89  917.87    98.6  916.59
   108.1  916.41   117.6   916.4     216   916.4   232.1   916.4   241.6  917.56
   251.2  921.34   260.7  926.89   270.2  932.31   279.6  937.84   316.8   959.9
   344.8  976.41   354.1  981.39   363.5  984.94   372.8  986.75   382.1  987.88
#Mann= 3 , 0 , 0
       0      .1       0    98.6    .045       0     216      .1       0
Bank Sta=98.6,216
XS Rating Curve= 0 ,0
Exp/Cntr=0.3,0.1

Type RM Length L Ch R = 1 ,1063.8  ,400.1,402.5,404.4
XS GIS Cut Line= 4
     1666331.413      745737.043     1666360.059       745760.48
     1666483.756      745920.636     1666561.881      746070.376
#Sta/Elev= 23
       0  949.62     9.2  945.22    18.5   940.5      37  930.96    56.3  920.76
    65.9  916.68    75.6  914.94    85.2   914.9   191.2   914.9   200.8   915.1
   210.5  916.47   220.1  920.08   239.4     928   248.8  932.06   267.5  940.34
   276.9  944.39   295.7  952.22   305.1     956   314.4  959.46   323.8  962.57
   342.6   968.4   370.7  976.91   408.3  988.05
#Mann= 3 , 0 , 0
       0      .1       0    75.6    .045       0   210.5      .1       0
Bank Sta=75.6,210.5
XS Rating Curve= 0 ,0
Exp/Cntr=0.3,0.1

Type RM Length L Ch R = 1 ,661.4   ,358.4,377.7,396.5
XS GIS Cut Line= 4
     1666084.017       745954.49     1666093.131      746043.032
     1666211.621      746226.626     1666281.934      746390.688
#Sta/Elev= 30
       0  943.16     8.9  941.81    35.6  937.24    44.5  935.41    71.2  929.14
     127  919.18   136.5  917.12     146   915.4   155.5  914.95     165   914.9
   269.5  914.92     279   915.1     286916.1979   288.5  916.59     298  920.13
   307.5  923.27   316.9  925.88   335.7  930.02   345.1  932.64   354.5  935.63
   363.9  938.31   373.3  941.74   382.7  944.86   410.9  953.86   429.6  960.13
     439  962.82   457.8  969.27   467.2  971.73   476.6   973.9     486  975.62
#Mann= 3 , 0 , 0
       0     .06       0   136.5    .045       0     286      .1       0
Bank Sta=136.5,286
XS Rating Curve= 0 ,0
Exp/Cntr=0.3,0.1

Type RM Length L Ch R = 1 ,283.7   ,234.1,249.7,265.2
XS GIS Cut Line= 4
     1665897.168      745995.723     1665840.744      746082.529
      1665766.96      746340.775      1665927.55      746542.598
#Sta/Elev= 30
       0  939.19     9.4  937.97    18.8  936.52    28.2  934.84    65.9  926.94
   103.5  920.03   113.1  917.98   122.7  915.48   132.3  914.84   141.9   914.8
   333.7  914.81     338915.0698   343.3  915.39   352.9  918.09   362.5  923.15
   372.1   927.5   381.7  930.41   410.3  938.12   429.4  942.44     439  944.85
   448.5  947.53   458.1  950.45   477.2  955.42   486.7  957.74   515.4  964.06
   534.5  968.88   563.2  976.73   591.8  985.19   610.9  990.65     630  995.72
#Mann= 3 , 0 , 0
       0     .06       0   122.7    .045       0     338      .1       0
Bank Sta=122.7,338
XS Rating Curve= 0 ,0
Exp/Cntr=0.3,0.1

Type RM Length L Ch R = 1 ,34      ,33.1,34,34.9
XS GIS Cut Line= 4
     1665783.401      745941.221     1665720.901      746028.026
     1665446.595      746229.415     1665189.651      746291.915
#Sta/Elev= 30
       0  943.49    68.1  930.27    87.5  926.32   136.1  915.81     144915.0765
   145.9   914.9   155.6   914.8   223.6  914.94   233.4  915.12   301.4  917.35
   340.3  917.68     350  917.69   388.9  916.58   408.4  915.83   418.1   916.4
     423918.1378   427.8  919.84   437.5  925.35   447.3  930.55   496.2  952.95
     506  956.78   515.8  959.67   525.6  961.36   545.2  963.76   564.8   965.8
   574.6  966.51   594.2  967.36   643.1     969   701.9  971.39   711.7  971.59
#Mann= 3 , 0 , 0
       0      .1       0     144    .045       0     423      .1       0
Bank Sta=144,423
XS Rating Curve= 0 ,0
Exp/Cntr=0.3,0.1

Chan Stop Cuts=-1
Use User Specified Reach Order=0
Composite Channel Slope=5
